--- SPLAURFK.prj (project) ---

Proj Title=SPLAURFK
Current Plan=p01
Default Exp/Contr=0,0
English Units
Geom File=g01
Flow File=f01
Plan File=p01
BEGIN DESCRIPTION:
END DESCRIPTION:
DSS Export Rating Curves= 0
DSS Export Rating Curve Sorted= 0
DSS Export Volume Flow Curves= 0
DXF OffsetX= 0
DXF OffsetY= 0
DXF ScaleX= 0
DXF ScaleY= 0

--- SPLAURFK.p01 (plan) ---

Plan Title=Floodplain
Program Version=4.00
Geom File=g01
Flow File=f01
K Sum by GR=0
Std Step Tol=0.01
Critical Tol=0.01
Num of Std Step Trials=20
Max Error Tol=0.3
Flow Tol Ratio=0.001
Split Flow NTrial=30
Split Flow Tol=0.02
Split Flow Ratio=0.02
Log Output Level=0
Friction Slope Method=1
Unsteady Friction Slope Method=2
Unsteady Bridges Friction Slope Method=1
Global Log Level=0
CheckData=False
Run HTab=0
Run UNet=0
Run PostProcess=0
UNET Theta=0
UNET Theta Warmup=0
UNET ZTol=0
UNET ZSATol=0
UNET MxIter=0
UNET MaxInSteps=0
UNET DtIC=0
UNET DtMin=0
UNET MaxCRTS=0
UNET WFStab=0
UNET SFStab=0
UNET WFX=0
UNET SFX=0
UNET DSS MLevel=0
UNET DZMax Abort=0
UNET Convert EG Bridges=0
UNET Use Existing IB Tables=0
UNET Froude Limit=0
UNET Froude Power=0
Write IC File=0
Echo Input=False
Echo Output=False
Write Detailed=0

--- SPLAURFK.f01 (steady flow) ---

Flow Title=NFF Regression Equation
Program Version=4.10
Number of Profiles= 1
Profile Names=P100yr
River Rch & RM=SPLAURFK,Main            ,83509.7
1046.105
River Rch & RM=SPLAURFK,Main            ,82009.7
1112.025
River Rch & RM=SPLAURFK,Main            ,81709.7
1218.976
River Rch & RM=SPLAURFK,Main            ,79909.7
1349.528
River Rch & RM=SPLAURFK,Main            ,76609.7
1776.607
River Rch & RM=SPLAURFK,Main            ,76309.7
1890.583
River Rch & RM=SPLAURFK,Main            ,72709.7
2065.322
River Rch & RM=SPLAURFK,Main            ,70009.7
2270.315
River Rch & RM=SPLAURFK,Main            ,61609.7
2522.399
River Rch & RM=SPLAURFK,Main            ,57109.7
2800.192
River Rch & RM=SPLAURFK,Main            ,51409.7
3673.811
River Rch & RM=SPLAURFK,Main            ,50809.7
3958.125
River Rch & RM=SPLAURFK,Main            ,42331.9
4380.245
River Rch & RM=SPLAURFK,Main            ,39109.7
4819.621
River Rch & RM=SPLAURFK,Main            ,29209.7
5153.663
River Rch & RM=SPLAURFK,Main            ,15409.7
5711.648
Boundary for River Rch & Prof#=SPLAURFK,Main            , 1
Up Type= 0
Dn Type= 1
Dn Known WS=816.65
DSS Import GetInterval= 0
DSS Import GetPeak= 0
DSS Import FillOption= 0

--- SPLAURFK.g01 (geometry) ---

Geom Title=USGS 10m DEM
Program Version=4.10

River Reach=SPLAURFK        ,Main
Reach XY= 30
     1765331.191        304893.2     1758891.955       305401.88
     1754141.065      309793.482     1751862.324      310858.187
     1752052.211      312941.303     1750380.119      316068.039
      1750778.34      321581.928     1753987.198      325400.439
       1754026.3      326887.092     1753003.135      327890.706
     1753332.894       329669.71     1752372.291      330589.255
     1754502.039      333764.586     1753030.506      334857.483
     1753326.376      336689.404     1751826.169      336910.982
     1751491.196      339547.359     1749417.898      338271.575
     1748603.669      340047.232     1746446.396      339441.631
     1746024.794       340710.64     1745007.732      340932.308
      1745457.53      344959.203     1744117.686      345003.473
     1744837.738      346510.114     1743831.227      347408.552
     1742077.321      346691.104     1739202.321      347766.494
     1739116.384      345329.385     1736734.873      344896.768

Type RM Length L Ch R = 1 ,83509.7 ,251.8,259.4,265.1
XS GIS Cut Line= 3
     1765307.846      304473.094     1765321.533      304895.791
     1765318.492      305150.301
#Sta/Elev= 30
       0 1677.25      20 1670.86    87.8 1641.66    99.7 1637.75   131.7 1620.49
   159.6 1612.17   179.5 1600.35   207.5 1587.52   227.4 1576.91   247.4  1560.1
   267.3 1558.44   335.1 1558.34   355.1 1554.47     387  1556.3     403 1553.56
   415.4 1548.24   422.9 1546.44   430.4 1547.06   442.8 1548.13   450.8 1551.46
   458.7  1558.1   470.6 1573.75   478.6 1580.55   506.4 1598.76   550.2  1621.7
     574 1631.49   613.8 1644.38   625.8 1645.83   645.6 1656.78   677.4 1667.08
#Mann= 3 , 0 , 0
       0      .1       0   415.4    .045       0   430.4      .1       0
Bank Sta=415.4,430.4
XS Rating Curve= 0 ,0
Exp/Cntr=0.3,0.1

Type RM Length L Ch R = 1 ,83250.2 ,296.7,287.2,277.6
XS GIS Cut Line= 4
     1765166.582      304544.833     1765142.323      304675.705
     1765081.946      304837.801     1764955.561      305255.043
#Sta/Elev= 30
       0 1675.26    19.6 1664.32    62.6 1644.84    97.9 1626.56   117.4 1610.98
   133.1 1605.29   148.8 1593.76   176.4 1578.76   203.9 1559.31   211.7 1555.51
   239.2 1549.55   262.8 1546.94   286.4 1546.64   298.2 1542.02   309.7  1541.2
   314.1 1540.92   324.7 1541.61   338.1 1545.26   358.1 1545.86   386.1 1549.69
   426.1 1575.82   442.1 1583.59   474.1 1602.84   534.1 1633.52     582 1656.04
     602 1667.01     622 1673.11     646 1684.62     698 1716.85     742 1740.85
#Mann= 3 , 0 , 0
       0      .1       0   309.7    .045       0   324.7      .1       0
Bank Sta=309.7,324.7
XS Rating Curve= 0 ,0
Exp/Cntr=0.3,0.1

Type RM Length L Ch R = 1 ,82963.1 ,362.1,353.4,344.9
XS GIS Cut Line= 3
      1764782.56      304409.739      1764819.36      304837.801
     1764875.117      305253.982
#Sta/Elev= 30
       0 1779.91    27.8 1761.11    47.7 1751.78    83.5 1725.36   151.2 1679.05
   167.1 1674.11   194.9 1659.69   222.8  1643.8   254.6 1622.17   278.5 1608.36
   334.2 1568.21   346.1 1558.53     362 1542.06   389.9 1537.66   424.1  1536.8
   433.6 1535.92   439.1 1536.08   453.6 1539.96   469.6 1537.19   525.6 1538.74
   541.6  1542.6   553.6 1550.06   589.6  1578.8   617.6 1598.22   629.6 1604.15
   669.6 1629.51   729.6 1661.07   777.6 1678.48   793.6 1689.01   849.5 1717.88
#Mann= 3 , 0 , 0
       0      .1       0   424.1    .045       0   439.1      .1       0
Bank Sta=424.1,439.1
XS Rating Curve= 0 ,0
Exp/Cntr=0.3,0.1

Type RM Length L Ch R = 1 ,82609.7 ,289.9,300,311
XS GIS Cut Line= 3
     1764351.152      304569.652     1764550.931      304974.504
     1764738.209      305330.323
#Sta/Elev= 30
       0  1716.9      44 1687.57    63.9 1670.58    67.9 1668.47    83.9 1665.19
   103.9 1653.95   127.8 1642.57   179.8 1606.91   191.8 1602.88   239.7 1576.63
   279.7 1559.12   339.6 1537.04   375.6  1534.9   411.5 1528.52   435.5 1530.49
     444 1528.51   455.4 1527.01   463.4 1528.81   475.4 1543.24   487.3 1561.26
   499.2 1573.06   511.2 1582.02     543 1601.86   574.9 1619.37   634.6 1647.44
   670.4    1658   686.4 1658.94   722.2  1672.5   801.8  1708.3   853.6 1728.95
#Mann= 3 , 0 , 0
       0      .1       0     444    .045       0   463.4      .1       0
Bank Sta=444,463.4
XS Rating Curve= 0 ,0
Exp/Cntr=0.3,0.1

Type RM Length L Ch R = 1 ,82309.7 ,296.1,300,302.6
XS GIS Cut Line= 4
     1764272.114      304590.856     1764276.879      305055.497
     1764273.178      305176.434      1764352.78      305323.912
#Sta/Elev= 30
       0 1713.37    31.8 1691.36    55.6 1672.54    71.5 1667.16    87.4 1656.41
   103.3 1650.68   123.1 1635.31   154.9 1615.89   174.8 1605.95   258.2 1550.73
     282 1542.32   309.8 1535.95   373.3 1528.94   436.9 1529.66   457.2 1521.02
   460.7 1520.28   472.2 1520.87   476.4 1522.48   480.3 1526.69   499.8 1555.28
   511.5 1567.65   566.1 1605.26   581.8 1609.09   593.6 1618.48   637.5  1642.1
   657.5 1652.25   677.4 1659.13   697.4 1668.78   721.3 1682.41   753.2 1703.61
#Mann= 3 , 0 , 0
       0      .1       0   457.2    .045       0   472.2      .1       0
Bank Sta=457.2,472.2
XS Rating Curve= 0 ,0
Exp/Cntr=0.3,0.1

Type RM Length L Ch R = 1 ,82009.7 ,301.2,300,297.8
XS GIS Cut Line= 3
     1764053.301       304662.02      1764008.17      304934.253
     1763941.856      305374.549
#Sta/Elev= 30
       0 1676.77      20  1662.8      40    1654      56 1649.27      72 1638.68
      84 1628.46     100 1622.55     140 1596.19     156 1583.34     168 1575.68
     196 1551.74     216  1536.9     240 1524.24     252 1521.75   268.4 1516.46
     276    1516   283.4 1516.93   291.8 1518.83   315.7 1521.53   331.6 1520.32
   343.5 1521.22     427 1532.54   446.9 1538.68   458.8 1545.33   470.8  1553.5
   502.6 1570.02   534.4 1579.84     598 1592.41   685.4 1607.45   721.2 1615.41
#Mann= 3 , 0 , 0
       0      .1       0   268.4    .045       0   283.4      .1       0
Bank Sta=268.4,283.4
XS Rating Curve= 0 ,0
Exp/Cntr=0.3,0.1

Type RM Length L Ch R = 1 ,81709.7 ,303.3,300,299.3
XS GIS Cut Line= 3
     1763772.208      304537.898     1763722.289      304974.473
     1763701.011       305378.42
#Sta/Elev= 30
       0 1751.35      36 1733.07   111.8 1679.57   155.8 1651.32   171.8 1646.35
   231.7 1608.38   247.7 1602.18   291.6 1568.58   323.6 1536.62   347.5 1515.82
   363.5 1513.03   423.4 1514.78   431.9 1510.79   439.4 1510.19   446.9 1510.83
   459.2 1514.93   494.9 1517.53   506.8 1524.06   534.6 1526.03   550.5 1537.49
   586.2 1555.98   665.5 1601.77   677.4 1611.06   697.2 1615.72   709.1 1624.64
   728.9 1635.58   756.7  1646.3   808.2  1672.5   820.1 1676.15   843.9 1691.39
#Mann= 3 , 0 , 0
       0      .1       0   431.9    .045       0   446.9      .1       0
Bank Sta=431.9,446.9
XS Rating Curve= 0 ,0
Exp/Cntr=0.3,0.1

Type RM Length L Ch R = 1 ,81409.7 ,296.9,300,299.8
XS GIS Cut Line= 3
     1763462.502      304489.125     1763480.319      304942.659
     1763467.185      305343.865
#Sta/Elev= 30
       0 1734.32    31.8 1711.85    83.6 1680.42   123.4 1658.44   139.4 1653.96
   159.3 1641.66   179.2 1635.25   191.1  1626.5     207 1618.89     223 1608.07
   238.9 1602.32   302.6 1565.08   318.5    1555   374.3 1510.43   378.2 1508.76
     426 1508.13   446.4 1504.64   453.9 1504.41   461.4 1504.96   477.7 1512.45
   493.6  1508.3   501.6 1508.82   509.5 1512.28   533.4 1517.54   561.2 1528.85
     740 1638.36   767.9 1651.61   779.8 1653.46   783.8 1655.79   855.3 1706.15
#Mann= 3 , 0 , 0
       0      .1       0   446.4    .045       0   461.4      .1       0
Bank Sta=446.4,461.4
XS Rating Curve= 0 ,0
Exp/Cntr=0.3,0.1

Type RM Length L Ch R = 1 ,81109.7 ,301.5,300,299.8
XS GIS Cut Line= 3
     1763289.095      304469.234     1763214.769      304874.465
     1763167.884      305208.895
#Sta/Elev= 30
       0 1661.44      20 1657.06      56 1645.98     100 1630.05     132 1615.88
     196 1580.88     216 1567.68     228 1562.69     248 1546.97     260 1540.85
     304 1505.65     316 1503.27     360 1501.45     388 1502.99   404.5 1496.92
     416 1496.41   419.5 1496.71   439.8 1500.15   455.7 1508.15   471.6 1518.81
   519.3 1559.56     551 1581.46     563 1587.39   578.8 1599.03   606.7 1614.06
   650.4 1642.91   670.2 1649.24   682.2  1655.7     706 1675.75   749.7 1707.17
#Mann= 3 , 0 , 0
       0      .1       0   404.5    .045       0   419.5      .1       0
Bank Sta=404.5,419.5
XS Rating Curve= 0 ,0
Exp/Cntr=0.3,0.1

Type RM Length L Ch R = 1 ,80809.7 ,311.4,300,288.6
XS GIS Cut Line= 3
     1762947.676      304439.391      1762925.88      304853.582
     1762905.297      305102.558
#Sta/Elev= 30
       0 1569.79    19.9 1564.13    43.9 1560.12    59.8 1554.64   103.7 1541.95
   135.6 1537.07   171.5 1527.88   179.5 1523.98   199.4 1512.06   211.4 1507.59
   227.3 1506.05   239.3 1506.41   255.2 1502.45   263.2  1502.9   307.1  1498.2
     331 1496.73   378.9 1495.97   407.3 1492.38   418.7 1491.64   426.7 1492.63
   434.6 1495.95   446.5 1497.53   470.3 1510.45   494.1 1525.05     506 1533.61
   517.9 1540.46   561.5 1569.91   573.4 1578.75     613 1602.35   664.6 1631.37
#Mann= 3 , 0 , 0
       0      .1       0   407.3    .045       0   426.7      .1       0
Bank Sta=407.3,426.7
XS Rating Curve= 0 ,0
Exp/Cntr=0.3,0.1

Type RM Length L Ch R = 1 ,80509.7 ,296.1,300,303.2
XS GIS Cut Line= 3
     1762519.012      304638.149     1762662.319      304941.478
     1762828.822      305315.197
#Sta/Elev= 30
       0 1605.07      28 1592.19    39.9 1583.96    71.9 1565.86    99.8 1546.97
   127.8 1530.57   139.8 1520.93   151.8 1518.15   167.7 1507.44   191.7  1496.8
   195.7  1495.4   207.7 1495.76   227.6 1493.89   279.6 1487.48   291.6 1488.03
   311.5 1491.01   315.5 1490.46     328 1484.93   331.5 1484.68     343 1484.73
   351.4 1486.46   510.2 1596.58   522.2 1603.41   585.7 1644.71   593.7 1647.64
   629.4 1672.67   665.2 1699.39   696.9 1720.41   712.8  1728.4   744.6 1750.16
#Mann= 3 , 0 , 0
       0      .1       0     328    .045       0     343      .1       0
Bank Sta=328,343
XS Rating Curve= 0 ,0
Exp/Cntr=0.3,0.1

Type RM Length L Ch R = 1 ,80209.7 ,301.9,300,299.9
XS GIS Cut Line= 3
     1762279.811       304667.73     1762389.261      305063.786
     1762501.838      305459.144
#Sta/Elev= 30
       0 1649.49    47.9 1624.06    67.8 1616.77    87.8 1601.87   119.7 1591.22
   139.6 1578.73   155.6 1576.56   211.4 1530.96   247.3 1496.51   251.3 1494.37
   295.2 1484.17   339.1 1482.96     355 1480.87   394.9 1481.76   403.4 1480.36
   410.9 1478.38   418.4  1478.4   422.9 1478.96   426.9 1481.66   434.8 1489.74
   446.8 1497.59   470.8 1517.24   486.7 1525.22   566.6 1579.39   598.5 1597.59
   638.4 1615.77   674.3 1629.92   722.2 1643.14   750.1 1647.51     822 1648.92
#Mann= 3 , 0 , 0
       0      .1       0   403.4    .045       0   418.4      .1       0
#XS Ineff= 2 , 0
          331.26 1490.24
Permanent Ineff=
       F       F
Bank Sta=403.4,418.4
XS Rating Curve= 0 ,0
Exp/Cntr=0.3,0.1

Type RM Length L Ch R = 1 ,79909.7 ,306.4,300,291.3
XS GIS Cut Line= 3
     1761975.796      304755.173     1762120.072      305149.955
     1762211.229      305550.547
#Sta/Elev= 30
       0 1714.86    19.8 1698.52     115  1636.8   126.9    1627   142.8 1621.38
   162.6 1610.75   202.2  1592.9   249.8 1560.05   293.4 1523.92   321.2  1503.6
     341 1486.23   352.9  1477.6   360.8 1475.49   384.6  1474.8   396.5 1477.14
   412.8 1474.25   424.3  1473.4   432.3 1474.44   444.2 1480.04   492.1 1484.75
   555.9 1497.41   571.9 1498.75   603.8 1496.64   611.8  1498.1   619.8 1501.95
   639.7 1515.93   667.6  1518.5   707.5 1534.63   779.3 1560.79   831.2  1583.3
#Mann= 3 , 0 , 0
       0      .1       0   412.8    .045       0   432.3      .1       0
Bank Sta=412.8,432.3
XS Rating Curve= 0 ,0
Exp/Cntr=0.3,0.1

Type RM Length L Ch R = 1 ,79609.7 ,291.5,300,310
XS GIS Cut Line= 3
     1761613.555      304895.001     1761855.866      305244.342
     1762091.081      305587.956
#Sta/Elev= 30
       0 1676.79    11.9 1671.14    35.8 1655.08    67.6 1655.79    71.5 1654.51
    87.4  1645.6   107.3 1637.33   139.1 1626.89     151 1624.65   162.9  1617.2
   174.8 1614.61   218.5 1595.91   242.4 1583.76   274.2 1564.69   309.9 1537.84
   321.8 1527.52   353.6 1492.25   373.5 1475.29   385.4 1469.11   393.4 1467.05
   432.7 1468.08     445  1470.8   472.7 1472.97   496.5 1471.87   540.2    1475
     564 1479.65   659.1 1534.78   758.3 1587.18   821.7 1613.86   841.6 1620.23
#Mann= 3 , 0 , 0
       0      .1       0   385.4    .045       0   432.7      .1       0
#XS Ineff= 2 , 0
                          471.45         1486.61
Permanent Ineff=
       F       F
Bank Sta=385.4,432.7
XS Rating Curve= 0 ,0
Exp/Cntr=0.3,0.1

Type RM Length L Ch R = 1 ,79309.7 ,293.8,300,302.4
XS GIS Cut Line= 3
     1761494.067      304943.201     1761595.275      305360.379
     1761667.007      305760.002
#Sta/Elev= 30
       0 1641.38    31.8 1620.95    55.6 1618.64    75.5 1607.46    95.4 1603.02
   107.3 1596.59   206.7 1560.93   222.6 1551.17   234.5 1539.48   250.4  1529.2
   286.2 1499.31     322 1477.42   349.8 1467.38   373.6 1464.86   389.5 1467.25
   413.4 1462.85   421.3 1462.51   433.3 1462.95     485 1468.44   508.9 1477.69
   552.7 1505.54   592.5  1538.7   644.2 1572.22     684 1593.89   731.8 1617.19
   747.7 1622.53   759.7 1629.91   775.6 1640.12   819.4 1672.85   835.3  1686.7
#Mann= 3 , 0 , 0
       0      .1       0   413.4    .045       0   433.3      .1       0
Bank Sta=413.4,433.3
XS Rating Curve= 0 ,0
Exp/Cntr=0.3,0.1

Type RM Length L Ch R = 1 ,79009.7 ,301.3,300,299.6
XS GIS Cut Line= 3
     1761316.755       305126.43     1761306.996      305338.688
     1761326.129      305775.967
#Sta/Elev= 30
       0 1546.06    35.4 1527.23    51.2  1517.6    82.6 1495.06    94.4 1487.95
   110.2 1474.69   125.9 1465.02   137.7 1461.66   165.3 1458.66   177.1 1460.04
     205 1457.05     220 1457.01   236.4 1460.02   276.2 1459.05     296 1461.95
     308 1470.09   335.8 1493.49   375.6 1524.67   435.3 1568.17   459.2 1583.78
     487 1597.19   522.8 1617.67   534.8 1621.55   538.8 1624.29   558.7 1638.76
   582.5 1664.66   590.5 1670.81   602.4 1675.73   614.4  1677.7   650.2 1676.37
#Mann= 3 , 0 , 0
       0      .1       0     205    .045       0     220      .1       0
Bank Sta=205,220
XS Rating Curve= 0 ,0
Exp/Cntr=0.3,0.1

Type RM Length L Ch R = 1 ,78709.7 ,269,268.3,267.4
XS GIS Cut Line= 4
     1761065.019      305048.305      1761052.69      305386.372
     1761041.368      305541.101     1761156.165      305629.902
#Sta/Elev= 30
       0 1575.07    19.9 1563.93    31.8 1555.67    51.7 1544.04    79.6  1520.5
    91.5 1512.52   115.4 1494.37   123.4 1490.75   139.3 1489.31   151.2 1485.33
   171.1 1468.16   179.1 1463.74     195 1460.15   226.8 1455.71   286.6  1458.2
   322.4 1454.58   330.8  1451.7   338.3 1449.88   350.2 1450.88   362.2 1454.92
   374.1 1464.25     390 1480.46   405.9 1490.07   417.8 1499.88   445.7 1516.74
   469.6 1526.03   493.4  1529.8   520.9 1542.55   575.8 1564.73   638.6 1584.17
#Mann= 3 , 0 , 0
       0      .1       0   330.8    .045       0   350.2      .1       0
#XS Ineff= 2 , 0
          275.41 1466.48
Permanent Ineff=
       F       F
Bank Sta=330.8,350.2
XS Rating Curve= 0 ,0
Exp/Cntr=0.3,0.1

Type RM Length L Ch R = 1 ,78441.4 ,320.1,331.7,345.1
XS GIS Cut Line= 3
     1760787.242      305056.985     1760787.242      305343.444
     1760774.193      305762.076
#Sta/Elev= 30
       0 1558.59       8 1553.11    39.8 1526.38    99.5 1480.84   115.4 1466.28
   135.3 1453.86   155.2 1451.21     195 1451.54   206.9 1450.08   222.8  1450.8
   262.6 1449.41   284.6 1445.54   294.4 1445.31   299.6 1445.81   310.4 1449.32
   330.3 1449.83   334.3 1452.41   346.3 1466.07   370.2 1483.13   386.2 1485.32
   398.2 1491.66   410.1 1495.28   426.1 1506.44   577.6 1575.49   597.6  1579.5
   609.6 1586.79   621.5 1591.68   657.4 1604.46   681.4 1611.05   705.3  1621.8
#Mann= 3 , 0 , 0
       0      .1       0   284.6    .045       0   299.6      .1       0
#XS Ineff= 2 , 0
          190.84  1461.9
Permanent Ineff=
       F       F
Bank Sta=284.6,299.6
XS Rating Curve= 0 ,0
Exp/Cntr=0.3,0.1

Type RM Length L Ch R = 1 ,78109.7 ,307.8,300,290.5
XS GIS Cut Line= 4
      1760613.63      305115.579     1760468.668      305345.238
     1760412.672      305422.796     1760394.446      305584.329
#Sta/Elev= 30
       0 1520.71       8 1515.65      24 1507.66    47.9 1490.83    63.9 1475.91
    79.9 1462.71   107.8 1445.98   111.8  1445.1   139.8 1445.03   167.7 1442.52
   199.7 1445.55   211.7 1444.35   227.6 1444.77   247.6 1443.24   264.1    1440
   271.6 1439.91   279.1 1440.21   287.5  1441.2   311.4 1447.89   323.4 1452.22
   335.4 1457.72   359.3 1462.03   363.3 1464.03   375.2 1474.94   387.1 1480.63
   402.9 1491.24   426.7 1504.05   482.2 1530.51   498.1 1536.38   529.8 1550.74
#Mann= 3 , 0 , 0
       0      .1       0   264.1    .045       0   279.1      .1       0
Bank Sta=264.1,279.1
XS Rating Curve= 0 ,0
Exp/Cntr=0.3,0.1

Type RM Length L Ch R = 1 ,77809.7 ,311.2,300,290.1
XS GIS Cut Line= 3
      1760290.28      305009.242     1760248.815      305242.457
     1760158.802      305642.547
#Sta/Elev= 30
       0 1571.42    23.7 1552.86    35.5 1545.77    63.2 1526.41    86.8 1512.02
   114.5  1497.3   134.2 1485.64     150 1472.15   169.8 1458.64   177.6 1451.69
   189.5 1438.97   193.4 1438.22   213.2 1438.55   229.4 1435.61   236.9 1434.45
   244.4  1435.9   252.8 1439.28   256.8  1439.7   316.5 1439.02   352.3 1442.15
   400.1 1442.94   404.1 1445.38     416 1455.11   467.8 1486.96   507.6 1515.24
   527.5 1527.54   567.3  1553.9   591.2 1566.21   615.1 1576.84     647 1587.41
#Mann= 3 , 0 , 0
       0      .1       0   229.4    .045       0   244.4      .1       0
Bank Sta=229.4,244.4
XS Rating Curve= 0 ,0
Exp/Cntr=0.3,0.1

Type RM Length L Ch R = 1 ,77509.7 ,299.2,300,297.5
XS GIS Cut Line= 3
     1759835.994      304802.361     1759960.155      305187.915
     1760034.203      305549.607
#Sta/Elev= 30
       0 1473.87     7.9 1473.29    15.9 1475.74    39.7 1489.15    55.6 1503.57
    67.5 1508.55    75.4 1509.22   107.2 1501.86   123.1  1495.9     131 1490.89
     143 1490.78   158.8 1483.86   198.6 1470.94     274 1453.12   313.7 1435.15
   345.5 1432.74   373.3 1434.38   397.6 1428.82     417 1428.12   420.9 1429.26
   432.8 1432.97   444.8 1430.47   460.6    1436   524.2 1435.91   555.9 1443.47
   571.8  1444.2   607.5 1449.97   643.2 1468.96   702.8 1507.09   774.2  1543.2
#Mann= 3 , 0 , 0
       0      .1       0   397.6    .045       0   420.9      .1       0
Bank Sta=397.6,420.9
XS Rating Curve= 0 ,0
Exp/Cntr=0.3,0.1

Type RM Length L Ch R = 1 ,77209.7 ,295.8,300,305.2
XS GIS Cut Line= 3
     1759570.141      304903.079     1759681.418      305297.481
     1759806.206      305687.449
#Sta/Elev= 30
       0 1476.16    63.7 1469.82   107.4 1450.63   127.3 1446.43   163.1 1448.12
     179 1442.81     187 1441.94     366 1425.49   389.9    1427   402.3 1424.64
   409.8 1423.45   421.7 1424.48   425.7 1426.99   453.5 1455.97   481.4 1479.61
   497.2  1486.6   509.2 1500.39     537 1521.93   572.8 1546.47   600.6 1560.54
   608.6 1562.69   624.5 1562.54   652.3 1556.85     704 1538.94   743.7 1519.34
   751.7 1522.12   763.6 1531.53   779.5 1540.22   791.4 1549.33   819.2 1563.95
#Mann= 3 , 0 , 0
       0      .1       0   402.3    .045       0   421.7      .1       0
Bank Sta=402.3,421.7
XS Rating Curve= 0 ,0
Exp/Cntr=0.3,0.1

Type RM Length L Ch R = 1 ,76909.7 ,298.6,300,299
XS GIS Cut Line= 4
     1759576.304      304761.846     1759356.342      305015.821
     1759383.795      305328.134     1759416.587      305736.561
#Sta/Elev= 30
       0 1520.79      12  1514.9      28 1510.75     104 1477.48     220 1433.03
   355.8 1426.05   435.2 1427.67     459  1424.3   498.7 1425.58     582 1421.02
   605.8  1423.7   633.6    1422     642  1418.5   645.5 1418.04     657  1418.2
   669.4 1422.13   697.2 1422.62   717.1 1443.03   768.8 1482.65   784.8 1491.59
   808.6 1512.23   828.5 1518.56   844.4 1534.77   880.2 1561.19   912.1 1578.41
     928 1589.48   943.9 1593.62   955.8 1603.27  1007.5 1636.37  1059.2 1664.62
#Mann= 3 , 0 , 0
       0      .1       0     642    .045       0     657      .1       0
Bank Sta=642,657
XS Rating Curve= 0 ,0
Exp/Cntr=0.3,0.1

Type RM Length L Ch R = 1 ,76609.7 ,310.8,300,293.4
XS GIS Cut Line= 3
     1759074.433      304941.698     1759084.925      305350.106
     1759135.311      305760.745
#Sta/Elev= 30
       0 1481.08    47.6 1460.66    83.3 1442.77   111.1  1430.9     119 1428.94
   218.2 1423.22   249.9 1419.64   313.4 1418.02   329.2 1415.68   392.7 1416.48
   396.6 1415.25   404.6 1412.85     416 1414.53   452.3 1416.24   460.3 1418.16
   464.2  1421.2   476.2 1436.78   496.1  1449.7     516  1466.1   531.9 1476.37
   567.7 1503.44   619.4 1545.22   635.3 1548.25   651.2 1558.18   671.1 1564.52
     683 1574.13   706.9 1582.02   714.8 1587.72   750.7 1604.23   822.3 1648.16
#Mann= 3 , 0 , 0
       0      .1       0   396.6    .045       0     416      .1       0
Bank Sta=396.6,416
XS Rating Curve= 0 ,0
Exp/Cntr=0.3,0.1

Type RM Length L Ch R = 1 ,76309.7 ,299.7,300,298.8
XS GIS Cut Line= 3
     1758612.247      305098.519     1758811.678      305458.711
       1758974.8      305833.892
#Sta/Elev= 30
       0  1527.7       8 1522.35      40 1495.74      52 1483.46      68 1474.82
    99.9 1447.67   135.9 1420.44   143.9 1416.37   179.9 1412.02   219.8  1411.1
   243.8 1413.48   263.8 1411.19   343.8 1410.05   391.7 1411.86   404.2 1408.99
   415.7 1408.01   419.2 1408.72   423.6 1412.37   435.6  1427.8   443.5 1435.82
   463.4 1449.13   499.1 1477.84   542.8 1505.96   594.4  1541.6   622.2 1558.71
   646.1 1569.39   681.8 1578.15   689.8 1583.34   745.4 1607.58   820.8 1647.72
#Mann= 3 , 0 , 0
       0      .1       0   404.2    .045       0   419.2      .1       0
Bank Sta=404.2,419.2
XS Rating Curve= 0 ,0
Exp/Cntr=0.3,0.1

Type RM Length L Ch R = 1 ,76009.7 ,298.2,300,300.2
XS GIS Cut Line= 3
     1758369.707      305267.489     1758562.385      305618.406
      1758748.43      305981.631
#Sta/Elev= 30
       0 1481.14    11.9 1473.14    27.8  1467.8    63.4    1445    99.1 1432.17
     115 1428.81   138.7 1421.18   166.5 1417.16   190.3 1411.12   202.2  1404.4
   269.5 1406.24   281.4 1403.28   293.3 1405.63   340.9 1406.84   376.6 1406.28
   392.8 1403.46   404.3 1403.04   407.8 1403.33   424.1 1414.06     440 1428.66
   471.6 1449.44   507.3 1476.23     543 1499.68   574.7  1522.6   626.2 1556.14
   638.1 1563.06   653.9 1566.84   697.5 1590.13     749 1620.33   808.4 1657.53
#Mann= 3 , 0 , 0
       0      .1       0   392.8    .045       0   407.8      .1       0
Bank Sta=392.8,407.8
XS Rating Curve= 0 ,0
Exp/Cntr=0.3,0.1

Type RM Length L Ch R = 1 ,75709.7 ,253.1,253.5,250.9
XS GIS Cut Line= 3
     1758127.683      305373.809     1758295.098       305747.59
     1758478.671      306115.287
#Sta/Elev= 30
       0 1551.31    31.8 1530.41    63.6 1505.35    87.5 1489.36   147.1 1441.18
     167 1430.89   178.9 1421.32   198.8 1401.82   206.8 1398.49   238.6 1397.22
   278.3  1403.5   310.2 1402.11   377.8 1402.28   393.7  1401.2   402.1 1399.26
   417.1 1398.62   453.4 1403.58   457.4 1406.19   469.4 1420.87   473.4 1424.65
   505.3 1445.03   541.2 1471.51   656.9 1552.88   680.9 1565.04   688.9 1567.59
   700.8 1569.29   712.8 1576.56   752.7 1592.43   764.7 1599.67   820.5 1640.81
#Mann= 3 , 0 , 0
       0      .1       0   402.1    .045       0   417.1      .1       0
Bank Sta=402.1,417.1
XS Rating Curve= 0 ,0
Exp/Cntr=0.3,0.1

Type RM Length L Ch R = 1 ,75456.2 ,347.1,346.5,349.4
XS GIS Cut Line= 3
     1757920.623      305493.811     1758083.249      305881.638
     1758301.601      306229.126
#Sta/Elev= 30
       0 1567.92    19.8 1556.52    59.5 1541.58    91.2 1521.62   107.1 1514.62
   130.9 1500.04   174.6 1479.58   222.2 1440.54     246 1430.28   281.7 1407.65
   305.5 1399.68   345.2 1395.27   396.7 1397.23   413.5 1395.03   424.5  1393.9
   428.5 1394.23   440.5 1398.17   468.4 1396.68   484.3 1403.36   512.2  1425.5
     556 1452.14     572 1465.54   619.8 1499.98   687.5 1545.18   719.4  1558.6
   735.3 1561.58   755.2 1573.77   787.1 1586.66     811 1598.75   830.9 1612.87
#Mann= 3 , 0 , 0
       0      .1       0   413.5    .045       0   428.5      .1       0
Bank Sta=413.5,428.5
XS Rating Curve= 0 ,0
Exp/Cntr=0.3,0.1

Type RM Length L Ch R = 1 ,75109.7 ,294.7,300,306.8
XS GIS Cut Line= 4
     1757633.955      305710.408     1757878.758      306128.434
     1757901.715      306169.846     1757994.273      306237.541
#Sta/Elev= 30
       0 1548.82    23.8 1543.12    43.7 1531.24    59.6 1518.37    79.4 1499.55
   119.1 1468.25     139 1450.11   154.9 1437.17   170.7 1427.17   198.5  1416.2
   214.4 1401.79   222.4 1397.72     270 1395.45   297.8 1392.36   341.5 1391.68
   353.4 1392.64   365.3 1390.69   385.2 1390.78     401 1392.25   416.9 1390.94
   440.8 1394.82   452.7 1392.29   476.9 1389.57   488.4 1388.46   496.3 1389.38
   508.1 1405.44   527.8 1422.26   555.5 1440.46   583.2 1457.21   646.4 1491.26
#Mann= 3 , 0 , 0
       0      .1       0   476.9    .045       0   496.3      .1       0
Bank Sta=476.9,496.3
XS Rating Curve= 0 ,0
Exp/Cntr=0.3,0.1

Type RM Length L Ch R = 1 ,74809.7 ,306.3,300,289.6
XS GIS Cut Line= 4
     1757521.183      305931.551     1757583.149       306135.17
     1757608.284      306264.854     1757673.092      306363.409
#Sta/Elev= 30
       0 1471.82    11.8 1463.37    23.6 1451.82    39.4 1439.69    78.8 1413.06
    86.7 1409.03    94.6 1403.11   106.4 1392.25   114.3 1387.85   126.1 1386.13
     138 1387.61   149.8 1387.98   173.4 1387.34   185.2 1385.25   205.3 1383.47
   208.9 1383.29   220.3 1383.54   232.3 1386.52   251.7 1386.53   267.2 1387.58
   282.8 1387.01   290.5 1388.68   325.5 1388.57     341  1389.9   352.8 1395.21
   368.5 1408.67   392.1 1425.53   403.9 1433.09   439.3 1449.04   462.9  1458.5
#Mann= 3 , 0 , 0
       0      .1       0   205.3    .045       0   220.3      .1       0
Bank Sta=205.3,220.3
XS Rating Curve= 0 ,0
Exp/Cntr=0.3,0.1

Type RM Length L Ch R = 1 ,74509.7 ,303.8,300,298
XS GIS Cut Line= 3
     1757236.894      306120.353     1757376.834      306273.605
     1757555.905      306469.746
#Sta/Elev= 30
       0 1489.42      16 1480.02    31.9 1473.55    43.9 1467.45    87.8 1440.55
    95.8 1434.88   111.8 1421.13   155.6 1386.95   159.6 1384.84   171.6 1381.44
   203.5  1379.2   215.5 1378.83   219.4 1379.11   239.2 1380.43   255.1 1384.11
     271 1383.65   286.8 1381.47   310.6 1381.89   330.4  1386.6   354.2  1389.1
   366.1 1384.02     374 1385.06     382 1389.39   389.9 1395.99   401.8 1409.85
   405.7 1412.94   417.6 1421.35   425.6 1425.71   437.4  1435.2   473.1 1459.46
#Mann= 3 , 0 , 0
       0      .1       0   203.5    .045       0   219.4      .1       0
#XS Ineff= 2 , 0
                          352.46         1398.17
Permanent Ineff=
       F       F
Bank Sta=203.5,219.4
XS Rating Curve= 0 ,0
Exp/Cntr=0.3,0.1

Type RM Length L Ch R = 1 ,74209.7 ,289.7,300,308.8
XS GIS Cut Line= 3
     1756950.518      306189.767     1757267.642      306541.305
     1757539.821      306831.908
#Sta/Elev= 30
       0  1522.3    11.9 1514.34    27.8 1512.62    35.8 1508.92    83.6  1477.1
   103.4 1460.85   115.4 1457.38   139.2 1440.82   234.7  1384.1   258.6 1380.66
   314.3 1383.15   326.2    1380   354.1 1383.31   381.9 1383.13   401.8 1379.34
   465.9  1377.1   480.9  1376.4   489.4 1377.36   493.4  1381.1   501.3 1396.83
   505.3  1402.3     569 1453.46   580.9 1462.35   592.9 1467.97   616.8 1487.23
   656.6 1506.29   688.4 1514.87   752.2 1522.81   835.8 1527.84   871.6 1526.46
#Mann= 3 , 0 , 0
       0      .1       0   465.9    .045       0   489.4      .1       0
Bank Sta=465.9,489.4
XS Rating Curve= 0 ,0
Exp/Cntr=0.3,0.1

Type RM Length L Ch R = 1 ,73909.7 ,379.2,372.6,370.2
XS GIS Cut Line= 3
     1756875.363      306223.661     1756994.331      306634.701
     1757095.835      306901.603
#Sta/Elev= 30
       0 1518.99      20  1517.1      24 1515.45      36 1504.96     100 1469.35
     112 1459.72     124 1456.04     140 1444.23     204 1402.55     236 1384.62
   279.9 1376.37   311.9  1375.4   331.9 1378.78   343.9 1377.22   387.9 1376.83
   403.9 1375.52   420.4 1371.91   427.9 1371.46   435.4 1371.55   475.5 1376.07
   499.3 1398.66     535 1422.65   554.8 1438.78   570.7 1449.46   590.5  1466.6
   602.4 1471.85   614.3 1482.02   657.9 1509.98   689.7 1527.49   713.5 1537.02
#Mann= 3 , 0 , 0
       0      .1       0   420.4    .045       0   435.4      .1       0
Bank Sta=420.4,435.4
XS Rating Curve= 0 ,0
Exp/Cntr=0.3,0.1

Type RM Length L Ch R = 1 ,73537   ,228.8,227.4,222.9
XS GIS Cut Line= 3
     1756557.641      306506.638     1756726.912      306769.225
     1756824.568      306975.388
#Sta/Elev= 30
       0 1420.87     7.9 1418.83    43.5 1401.49    63.3 1389.75    75.1 1386.48
      91 1378.96    98.9  1376.8   118.6 1374.79   146.3 1374.45   162.1 1372.11
   217.5 1370.65   229.4 1369.16   253.1  1370.3     265 1369.26   300.6 1368.94
   309.8 1366.69   312.4 1365.32   320.3 1364.32   324.8 1364.54     336 1364.99
   343.9 1368.81   359.6 1385.63   371.4 1395.76   430.4 1437.06   461.9 1460.54
   477.6 1473.72   485.5  1476.6   505.1 1492.54   520.9 1502.56   540.5 1517.96
#Mann= 3 , 0 , 0
       0      .1       0   309.8    .045       0   324.8      .1       0
Bank Sta=309.8,324.8
XS Rating Curve= 0 ,0
Exp/Cntr=0.3,0.1

Type RM Length L Ch R = 1 ,73309.7 ,257,247.5,235.7
XS GIS Cut Line= 3
     1756320.995      306583.891     1756555.527      306919.859
     1756796.998      307251.873
#Sta/Elev= 30
       0 1399.96    51.7 1393.49    83.5 1394.95    99.4 1399.16   115.4 1400.17
   123.3 1398.19   147.2 1385.15   163.1 1381.54     175 1375.29     183 1373.52
   230.7  1369.9   282.4 1368.83   306.3 1364.18   330.2 1366.75   381.9 1365.78
   402.2 1361.04   405.8 1361.01   417.2 1361.38   441.6  1366.4   445.6 1369.41
   453.6 1381.22   457.6 1384.98   501.4 1415.48   513.4 1426.54   565.2 1464.95
   632.9 1507.29   644.9 1513.67   696.7 1527.93   760.5 1554.16   820.3 1589.79
#Mann= 3 , 0 , 0
       0      .1       0   402.2    .045       0   417.2      .1       0
Bank Sta=402.2,417.2
XS Rating Curve= 0 ,0
Exp/Cntr=0.3,0.1

Type RM Length L Ch R = 1 ,73062.1 ,357.3,352.5,349.9
XS GIS Cut Line= 3
     1756104.082      306899.433     1756360.158      307064.364
      1756546.79       307159.85
#Sta/Elev= 30
       0 1414.02    19.8 1403.16    39.6 1388.88    55.4  1379.7    63.3  1375.8
    71.2  1373.9    83.1 1368.68   102.8 1367.34   118.7 1368.01   138.4 1367.58
   189.9 1363.84   233.4 1364.79   245.3 1361.57   261.1 1360.49   288.1 1357.06
   288.8 1357.03   303.1  1357.6   312.5 1360.63   320.4 1361.67   340.2 1362.03
     360    1360   363.9  1361.6   391.6 1384.13   407.4 1392.56   419.3 1401.46
   486.6 1445.95   498.4  1455.2   502.4 1457.62   510.3 1460.34   514.2 1463.18
#Mann= 3 , 0 , 0
       0      .1       0   288.1    .045       0   303.1      .1       0
Bank Sta=288.1,303.1
XS Rating Curve= 0 ,0
Exp/Cntr=0.3,0.1

Type RM Length L Ch R = 1 ,72709.7 ,240.4,243,245.1
XS GIS Cut Line= 3
     1755901.771      307227.628     1756286.624      307372.792
     1756670.856      307513.478
#Sta/Elev= 30
       0 1478.47    35.9 1451.64    63.9 1427.97    79.9  1416.3    99.8 1397.21
   111.8  1388.7   139.8 1362.56   147.8 1356.71   155.7 1355.38   187.7 1357.49
   239.6 1356.77   267.6  1359.3   299.5  1359.9   359.4 1357.75   379.4 1360.29
   403.8 1352.94   407.3 1352.76   418.8 1353.12   427.2  1356.1   447.1 1376.97
   490.8 1413.36   514.6 1427.27   526.5 1437.88   617.9 1500.68   637.8 1510.37
   685.4 1524.86   733.1  1547.8     753 1559.17   776.8 1575.25   820.5  1606.9
#Mann= 3 , 0 , 0
       0      .1       0   403.8    .045       0   418.8      .1       0
Bank Sta=403.8,418.8
XS Rating Curve= 0 ,0
Exp/Cntr=0.3,0.1

Type RM Length L Ch R = 1 ,72466.7 ,359.3,357,354.3
XS GIS Cut Line= 3
     1755826.304      307407.246     1756162.676      307578.687
     1756351.478      307669.833
#Sta/Elev= 30
       0 1489.59    11.9 1481.84    67.6 1439.17   103.3 1406.17   111.3 1401.28
   123.2 1391.07   143.1 1376.26     159 1360.94   174.9 1351.68   186.8 1350.86
   230.5  1354.5   246.4  1352.6   254.3 1354.02   329.8 1355.54   341.8 1353.29
   353.7 1353.34   373.6  1350.3   381.5 1350.11   393.4 1351.41   409.2 1356.76
     421 1365.32   436.9 1379.93   452.7 1391.57   460.6 1398.62   472.5 1402.93
   480.4 1410.18   496.2 1420.98   539.7 1448.54   555.6 1456.56   587.2 1480.33
#Mann= 3 , 0 , 0
       0      .1       0   373.6    .045       0   393.4      .1       0
Bank Sta=373.6,393.4
XS Rating Curve= 0 ,0
Exp/Cntr=0.3,0.1

Type RM Length L Ch R = 1 ,72109.7 ,358.7,362.6,368.2
XS GIS Cut Line= 3
     1755717.797      307739.277     1755907.476      307811.152
      1756227.78      307912.888
#Sta/Elev= 30
       0 1456.24    19.9 1441.48    51.7 1420.98    75.6 1401.65    91.5 1391.48
   111.4 1376.09   123.3 1369.44   143.2  1352.4   147.2 1350.19   163.1 1345.34
   195.3 1345.21   202.8 1344.91   210.3 1345.61   218.7 1347.37   230.5 1346.42
   254.2 1350.29   281.9 1351.68   297.7 1352.03   309.6 1351.18   345.2 1352.27
   388.7 1350.13   400.5 1351.82   404.5 1353.32   412.4 1358.28   424.2 1367.93
   432.2 1377.16   436.1 1380.73     448 1388.71   487.5 1418.84   538.9  1455.1
#Mann= 3 , 0 , 0
       0      .1       0   195.3    .045       0   210.3      .1       0
Bank Sta=195.3,210.3
XS Rating Curve= 0 ,0
Exp/Cntr=0.3,0.1

Type RM Length L Ch R = 1 ,71747.1 ,232.8,237.4,244.1
XS GIS Cut Line= 3
     1755620.141      307960.631     1755954.342      308160.284
     1756104.082       308257.94
#Sta/Elev= 30
       0 1437.19     7.9 1433.81    15.9 1428.64    27.8  1417.6    43.7  1405.4
    59.6 1388.99    71.5 1382.69    75.5 1379.63    99.3  1358.6   115.2 1349.24
   135.1 1342.86     143 1341.47   162.9 1344.02   210.5 1342.56   266.2 1343.46
   349.6 1341.79   369.4  1342.7   381.9  1341.3   397.2 1340.01   401.2 1340.41
   405.2 1342.96   409.2 1347.96   417.1 1363.15     425 1373.57     437  1385.3
   448.9 1394.82   472.7 1415.73   488.6 1427.22   544.2 1462.29   568.1 1474.91
#Mann= 3 , 0 , 0
       0      .1       0   381.9    .045       0   405.2      .1       0
Bank Sta=381.9,405.2
XS Rating Curve= 0 ,0
Exp/Cntr=0.3,0.1

Type RM Length L Ch R = 1 ,71509.7 ,295.2,300,300.1
XS GIS Cut Line= 3
     1755459.843      308019.258     1755773.176      308305.663
     1756032.631      308619.051
#Sta/Elev= 30
       0 1491.92    15.9 1485.41    59.5 1455.19    75.4 1446.89   138.9 1403.11
   166.6 1380.27   182.5  1371.8   206.3 1352.14   218.2 1346.16   230.1 1344.11
     242 1339.29   261.8 1342.17   301.5 1342.97   321.4 1341.32   345.2 1341.77
   357.1 1339.04   396.7 1340.78   408.6 1336.58   420.5 1336.15     432 1337.17
   460.4 1338.98   480.4 1343.26   508.3 1369.57   540.2 1388.73     588 1413.24
   663.8 1443.64   727.6 1460.55   787.5 1461.02   815.4 1469.08   831.4 1478.74
#Mann= 3 , 0 , 0
       0      .1       0   408.6    .045       0     432      .1       0
#XS Ineff= 2 , 0
          282.08 1351.93
Permanent Ineff=
       F       F
Bank Sta=408.6,432
XS Rating Curve= 0 ,0
Exp/Cntr=0.3,0.1

Type RM Length L Ch R = 1 ,71209.7 ,279.6,277.8,278.2
XS GIS Cut Line= 3
      1755290.75      308142.333     1755527.438      308475.584
     1755788.784      308795.271
#Sta/Elev= 30
       0 1482.34    35.7 1467.22    47.6 1459.46    63.5 1451.85   107.2  1424.5
     119 1414.65     131 1409.64   170.6 1380.77   234.1 1342.13   269.8 1336.48
   289.7 1339.69   357.2  1335.6   392.9 1335.04   401.2 1332.48   408.8 1332.14
   416.2 1332.23   444.5 1335.49     504 1336.72     508 1338.64     516 1345.59
   523.9 1357.65   531.8 1366.61   555.6 1384.58   575.5 1394.74   587.4  1398.9
   635.1 1410.58   662.8 1415.45   690.6 1424.14   766.1 1438.55   821.7 1454.46
#Mann= 3 , 0 , 0
       0      .1       0   401.2    .045       0   416.2      .1       0
#XS Ineff= 2 , 0
          293.39 1347.43
Permanent Ineff=
       F       F
Bank Sta=401.2,416.2
XS Rating Curve= 0 ,0
Exp/Cntr=0.3,0.1

Type RM Length L Ch R = 1 ,70931.8 ,316.2,322.2,326.6
XS GIS Cut Line= 4
     1755153.561      308359.937     1755146.474      308449.676
     1755316.321      308642.055     1755431.339      308778.774
#Sta/Elev= 30
       0 1386.28    11.7  1380.8    74.4 1355.79    86.1 1350.34      90 1349.01
   117.7 1345.53   145.3 1335.55   157.1 1334.91   176.9 1335.38   192.7 1334.57
   204.5 1332.84   224.2 1332.52     240 1333.45   271.6 1331.95   311.1 1332.28
     323 1331.73   334.8 1328.84   340.8 1328.18   350.6 1327.65   355.8 1327.95
   374.4 1330.69   394.3 1329.71   402.2 1332.59   406.2 1335.86   418.1 1352.95
   422.1 1356.55     438 1367.38   453.8  1380.2   493.6  1408.8   525.3 1429.14
#Mann= 3 , 0 , 0
       0      .1       0   340.8    .045       0   355.8      .1       0
Bank Sta=340.8,355.8
XS Rating Curve= 0 ,0
Exp/Cntr=0.3,0.1

Type RM Length L Ch R = 1 ,70609.7 ,306,300,295.4
XS GIS Cut Line= 3
     1754880.927      308448.473      1755057.67      308819.603
      1755248.17      309181.694
#Sta/Elev= 30
       0 1360.16    43.9 1367.32    75.8 1366.96   103.8 1363.12   171.6 1343.99
   203.5 1342.98   223.5 1333.16   255.4 1334.95   267.4 1331.22   347.2 1326.83
   363.2 1324.05   383.1 1325.14   399.1 1322.79   403.6 1322.81   418.6 1323.01
   438.9 1331.05   450.8 1341.18   474.6 1365.88   506.4    1391   538.2 1413.27
   573.9  1440.6   581.9 1445.34   601.7 1461.15   633.5 1474.32   649.4 1479.12
   669.3 1489.48   685.2 1500.71     713 1515.08   764.6 1553.14   820.2 1583.86
#Mann= 3 , 0 , 0
       0      .1       0   403.6    .045       0   418.6      .1       0
Bank Sta=403.6,418.6
XS Rating Curve= 0 ,0
Exp/Cntr=0.3,0.1

Type RM Length L Ch R = 1 ,70309.7 ,298.8,300,299.8
XS GIS Cut Line= 3
     1754557.534      308673.014     1754819.089      308987.836
     1754925.696      309123.826
#Sta/Elev= 30
       0 1435.18    11.9 1426.83    23.8 1415.46    43.7 1411.38    55.6 1401.88
    71.5 1393.39    87.4 1377.17   103.3 1365.65   111.3 1363.14   123.2 1363.25
   127.2 1361.71     151 1344.46   174.8 1334.95   206.6 1329.94   254.3 1326.23
     302 1326.83   317.9 1324.67   349.7 1324.08   361.6 1321.13   389.4 1321.85
   401.8 1320.45   409.3 1320.15   416.8  1320.5   432.9 1320.82   440.7 1323.87
   444.6 1326.37   464.3 1347.07   491.8  1367.2   554.6 1405.23   582.1 1417.95
#Mann= 3 , 0 , 0
       0      .1       0   401.8    .045       0   416.8      .1       0
Bank Sta=401.8,416.8
XS Rating Curve= 0 ,0
Exp/Cntr=0.3,0.1

Type RM Length L Ch R = 1 ,70009.7 ,303.4,300,296.8
XS GIS Cut Line= 3
     1754363.305      308866.161     1754607.109       309195.41
     1754859.764      309517.633
#Sta/Elev= 30
       0 1465.66    15.9 1454.82    27.8 1453.02    31.8  1450.6    59.7 1430.17
    75.6  1412.4    83.5 1409.16    99.4 1407.91   155.1 1359.59     187 1336.61
   206.8 1326.19   242.6 1322.58   254.6 1317.96   342.1 1322.18     354 1320.82
   365.9 1316.42   385.8 1318.13   402.2 1316.45   413.7 1316.14   417.2 1316.26
   453.4 1320.65   497.2 1353.32     517  1362.6   592.6 1389.49   652.2 1415.84
   668.1 1420.96   711.8 1444.65   735.7 1454.63   803.2 1473.08   819.2 1479.18
#Mann= 3 , 0 , 0
       0      .1       0   402.2    .045       0   417.2      .1       0
Bank Sta=402.2,417.2
XS Rating Curve= 0 ,0
Exp/Cntr=0.3,0.1

Type RM Length L Ch R = 1 ,69709.7 ,302.8,300,292.4
XS GIS Cut Line= 4
     1754086.624      309098.646     1754378.164      309386.272
     1754485.915      309489.879     1754639.238      309553.513
#Sta/Elev= 30
       0 1543.95    43.7 1509.98    59.6  1500.5    71.6 1490.73    87.5 1482.52
   111.3 1464.13   119.3 1460.87   143.1 1461.09     163 1446.27   186.9 1433.32
   238.6 1397.06   290.3 1356.93   302.2 1346.27   318.1  1340.4     342 1318.39
   361.8 1316.11   377.7 1312.21     402 1312.21     417 1311.48   429.2 1312.07
   444.9  1316.3   527.6 1315.97   547.2 1318.54     559 1321.59   586.7 1333.31
   602.5 1344.53     646 1368.85   673.6 1382.24   701.3 1397.59     725 1408.52
#Mann= 3 , 0 , 0
       0      .1       0     402    .045       0     417      .1       0
Bank Sta=402,417
XS Rating Curve= 0 ,0
Exp/Cntr=0.3,0.1

Type RM Length L Ch R = 1 ,69409.7 ,291,300,313.5
XS GIS Cut Line= 3
     1753840.319      309346.907     1754165.627      309594.104
     1754566.152      309779.897
#Sta/Elev= 30
       0  1463.7   107.1 1439.86   138.8  1426.9   150.7  1418.6   182.5  1409.2
   198.3 1398.18   218.2 1388.93   249.9  1370.4   289.6 1351.14   317.3 1333.14
   345.1 1318.69     357  1313.8   388.7 1315.39   401.1 1309.19   408.6 1307.58
   416.1 1307.84   436.4 1310.25   472.2 1311.55   488.1 1310.48   523.9 1313.67
   583.6 1310.72   603.5 1314.51   611.4 1318.46   639.3 1337.35   706.9 1392.05
   726.8    1405   746.7 1415.41   774.5 1425.05   830.2 1450.59   850.1 1457.62
#Mann= 3 , 0 , 0
       0      .1       0   401.1    .045       0   416.1      .1       0
Bank Sta=401.1,416.1
XS Rating Curve= 0 ,0
Exp/Cntr=0.3,0.1

Type RM Length L Ch R = 1 ,69109.7 ,290.4,300,311.5
XS GIS Cut Line= 4
     1753916.582      309427.645     1753919.929      309610.534
      1754053.76      309833.243     1754122.745      309944.138
#Sta/Elev= 30
       0 1431.66    15.9 1426.36    31.8 1418.54    71.6  1392.6    87.5 1380.27
   103.4 1370.95   115.3 1361.32   131.2  1352.5   139.2 1345.93     175 1321.72
   182.9  1317.1   194.9 1313.01   214.9 1312.56   230.9 1315.14   246.9 1312.64
   270.9 1314.74   290.8 1309.94   350.8 1308.36   398.8 1309.69   422.8 1307.54
   434.8  1304.6   438.8 1304.55   450.2 1304.95   458.6 1305.51   462.5 1307.39
   474.4 1323.23   482.3 1331.05   494.2 1338.82   533.8 1371.57   573.4 1397.38
#Mann= 3 , 0 , 0
       0      .1       0   434.8    .045       0   450.2      .1       0
Bank Sta=434.8,450.2
XS Rating Curve= 0 ,0
Exp/Cntr=0.3,0.1

Type RM Length L Ch R = 1 ,68809.7 ,298.3,300,300.2
XS GIS Cut Line= 3
     1753714.127       309413.12      1753758.64      309829.807
     1753769.012      310030.944
#Sta/Elev= 30
       0  1437.9    39.9 1419.55   103.8  1377.2   179.6 1329.69   191.6 1322.93
   211.5 1313.61   247.4 1307.21   263.4 1308.13   275.4 1310.54   283.4 1309.28
   303.3 1309.02   315.3 1304.43   323.3 1303.21   387.1 1305.53   391.1 1305.27
   403.1  1301.4   411.6 1300.63     423  1300.5   426.6 1300.79   446.7 1304.23
   454.6 1304.55   458.6 1305.47   462.5 1307.76   478.3 1326.24   494.1 1337.33
   513.8 1354.35     581 1398.51   592.8 1407.73   604.7 1414.63   620.5 1425.35
#Mann= 3 , 0 , 0
       0      .1       0   411.6    .045       0   426.6      .1       0
Bank Sta=411.6,426.6
XS Rating Curve= 0 ,0
Exp/Cntr=0.3,0.1

Type RM Length L Ch R = 1 ,68509.7 ,240,237.1,234.3
XS GIS Cut Line= 3
     1753443.492      309449.346     1753461.508      309838.054
     1753477.919      310250.213
#Sta/Elev= 30
       0 1377.31     7.9 1375.34    19.8 1369.04    63.5 1352.05    95.3 1344.51
   150.9  1327.7   166.8 1315.75   182.6  1313.3   198.5 1302.56   202.5  1301.4
   337.5 1302.21   381.6 1297.54   393.1 1297.46   396.6 1297.68     409 1301.12
   436.7 1321.08   456.6 1329.79   468.4 1340.03   484.3 1351.58   504.1 1360.56
   527.9 1376.82   571.6 1403.72   615.2 1433.66   631.1 1439.21   650.9 1448.37
   686.6  1458.6   706.4 1470.43   742.1  1487.4   773.8 1512.85   801.6 1532.59
#Mann= 3 , 0 , 0
       0      .1       0   381.6    .045       0   396.6      .1       0
Bank Sta=381.6,396.6
XS Rating Curve= 0 ,0
Exp/Cntr=0.3,0.1

Type RM Length L Ch R = 1 ,68272.6 ,363.9,362.9,361.4
XS GIS Cut Line= 3
     1753176.565       309505.77     1753228.648      309798.739
     1753276.391      310087.367
#Sta/Elev= 30
       0  1384.1       4 1381.07    19.8 1365.94    39.7 1348.41    67.4  1329.2
    79.4  1318.7    91.2 1311.87    99.2 1308.41     123 1301.82   130.9 1300.66
   174.6 1299.94   202.3 1298.31   210.3 1298.24   222.2 1299.86     250 1298.22
   269.8 1298.91   273.8 1298.63   285.7 1295.28   297.6 1294.46   305.5 1294.85
   325.2 1297.59   412.2  1295.8   416.2 1298.39   424.1 1306.06   435.9 1319.29
   439.9 1322.34   558.5 1399.11   566.4 1404.56   582.2 1417.52   590.1 1422.36
#Mann= 3 , 0 , 0
       0      .1       0   285.7    .045       0   305.5      .1       0
Bank Sta=285.7,305.5
XS Rating Curve= 0 ,0
Exp/Cntr=0.3,0.1

Type RM Length L Ch R = 1 ,67909.7 ,301.7,300,294
XS GIS Cut Line= 3
     1752871.148      309535.832     1752969.878      309942.633
     1753024.655      310152.471
#Sta/Elev= 30
       0 1426.91      16 1416.72    51.8 1389.42    79.7  1361.8    95.7 1354.26
   115.6 1334.04   119.6 1331.07   139.5 1324.56   147.5  1319.7   167.4  1303.4
   175.4 1298.78   199.3 1293.99   263.1 1296.74     303  1294.8   318.9 1295.99
   334.9 1293.66   354.8  1296.1   382.7 1296.13   394.7 1294.66   402.7  1289.6
   410.6 1289.46   411.1 1289.48   426.1 1289.55   442.3  1292.2   465.9 1291.95
   469.9 1293.28   485.6 1310.51   513.2 1331.97   544.8 1354.52   635.5 1413.23
#Mann= 3 , 0 , 0
       0      .1       0   411.1    .045       0   426.1      .1       0
Bank Sta=411.1,426.1
XS Rating Curve= 0 ,0
Exp/Cntr=0.3,0.1

Type RM Length L Ch R = 1 ,67609.7 ,306.9,300,299.7
XS GIS Cut Line= 3
     1752557.978      309640.305     1752691.443      310034.241
     1752891.387      310390.309
#Sta/Elev= 30
       0 1402.54      24 1385.25      32 1376.76      44 1374.86      96 1337.89
     160 1298.14     180 1292.91     236 1292.74     256  1290.3     292 1292.47
     312 1288.96     328  1291.9   343.9 1289.29   351.9 1291.06   375.9 1291.01
   408.4 1284.95   419.9  1284.4   423.4 1284.44   431.8    1285   439.7 1288.73
   459.5 1309.04   479.4 1325.64   558.7 1376.39   586.4 1396.39   618.1  1411.5
   649.8 1431.37   665.7 1438.45   713.3 1454.42   796.5 1474.48   824.3 1488.56
#Mann= 3 , 0 , 0
       0      .1       0   408.4    .045       0   423.4      .1       0
Bank Sta=408.4,423.4
XS Rating Curve= 0 ,0
Exp/Cntr=0.3,0.1

Type RM Length L Ch R = 1 ,67309.7 ,306.4,300,291.5
XS GIS Cut Line= 3
     1752169.479      309771.646     1752405.423      310100.905
     1752617.893      310479.687
#Sta/Elev= 30
       0 1392.16    27.8 1374.08    47.7 1365.76    63.5 1356.57   127.1 1327.92
   166.8 1312.64   178.7 1305.87   190.6 1302.27   222.4 1286.86   385.2 1284.53
   397.6 1281.32     409 1281.23   412.6 1281.28     429 1282.98   444.9 1282.07
   464.8 1284.36   472.8 1287.49   480.8 1295.19   492.7 1309.54   504.7 1320.04
   520.6  1330.4   532.6 1340.98   552.5 1354.57   652.1 1430.38     668 1439.95
     684 1445.86   699.9 1454.18   747.7 1480.55   819.4 1534.81   839.4  1546.5
#Mann= 3 , 0 , 0
       0      .1       0   397.6    .045       0   412.6      .1       0
Bank Sta=397.6,412.6
XS Rating Curve= 0 ,0
Exp/Cntr=0.3,0.1
