HEC-RAS study SPLAURFK.prj: SPLAURFK

--- SPLAURFK.g01 (geometry) --- (continued)

Type RM Length L Ch R = 1 ,33179.6 ,393.1,370,348.1
XS GIS Cut Line= 5
     1752250.132      336406.595     1752170.617      336522.878
     1752173.743      336852.775     1752168.535      337113.192
     1752345.618      337199.997
#Sta/Elev= 30
       0 1054.21     7.8 1049.43    31.3 1038.42      47 1028.49    78.3 1012.71
   121.3  995.07   140.9  992.85   156.8   989.7   216.4  983.89   387.3   977.6
   419.1  977.65   468.9  967.24   478.7  966.96   483.9     967   498.4  968.96
   518.1  978.45   522.1  979.05   597.1  978.21   628.6  982.33   660.2  982.97
     672  982.01   683.9  988.19   699.7 1003.33   727.3 1022.67     751 1045.25
   762.8 1053.04     818  1076.9   861.4 1090.76   877.2 1091.52   928.5 1102.45
#Mann= 3 , 0 , 0
       0    .006       0   468.9    .045       0   483.9      .1       0
#XS Ineff= 2 , 0
                          549.46          986.86
Permanent Ineff=
       F       F
Bank Sta=468.9,483.9
XS Rating Curve= 0 ,0
Exp/Cntr=0.3,0.1

Type RM Length L Ch R = 1 ,32809.7 ,437.1,430.3,423.8
XS GIS Cut Line= 3
     1751516.979      336713.489     1751830.503      336903.843
     1752180.688      337156.595
#Sta/Elev= 30
       0 1142.24    35.9 1113.71    47.8 1108.66    75.8 1089.09    91.7 1084.29
   127.6 1057.58   167.4 1019.36   191.4  986.44   207.3  973.48   239.2  971.56
   255.2  975.85   271.1  970.72     287  973.85   338.9  973.59   359.3   965.7
   370.8  965.52   374.3  965.61   398.8  968.25   430.8  975.62   514.7  973.63
   594.7  976.54   646.7  975.06   694.7     982   710.7  981.14   718.7  985.74
   734.7 1001.78   750.7  1012.3   770.7 1038.55   782.7 1046.73   798.7 1052.71
#Mann= 3 , 0 , 0
       0     .08       0   359.3    .045       0   374.3      .1       0
#XS Ineff= 2 , 0
                          554.89          990.48
Permanent Ineff=
       F       F
Bank Sta=359.3,374.3
XS Rating Curve= 0 ,0
Exp/Cntr=0.3,0.1

Type RM Length L Ch R = 1 ,32379.3 ,174.7,169.7,164.5
XS GIS Cut Line= 4
     1751508.784      337158.749     1751606.441      337175.676
     1751935.075      337252.614     1752120.764      337314.999
#Sta/Elev= 30
       0 1055.54    59.5 1007.29    87.2  981.35    95.2   974.8    99.1  972.68
     111  972.89   146.8  971.02     254  969.59   301.6  970.21   333.4  969.14
   369.1  969.84   408.8  966.61   429.1  961.15   436.6  960.62   444.1  960.95
   452.6  961.95   456.6  963.76   460.6   966.9   468.6  976.52   472.6  978.91
   488.6  980.61   504.6  979.81   520.6  986.76   524.6  988.83   532.6  995.21
   540.6 1005.59   548.6 1013.45   552.6 1016.32   556.6 1017.89   632.5 1029.98
#Mann= 3 , 0 , 0
       0      .1       0   429.1    .045       0   444.1      .1       0
Bank Sta=429.1,444.1
XS Rating Curve= 0 ,0
Exp/Cntr=0.3,0.1

Type RM Length L Ch R = 1 ,32209.7 ,298.6,300,300.4
XS GIS Cut Line= 3
      1751494.32      337414.603     1751905.227       337418.31
     1752312.651      337457.024
#Sta/Elev= 30
       0  1034.4    35.9 1004.63    55.8  985.26    71.8  974.36    79.8  971.58
   151.6  968.91   359.1  969.44     379  967.23     391  960.93     399  960.24
   403.4  960.36   418.4     961   426.8  965.12   438.7  975.91   442.7   978.1
   458.6  979.58   470.5  978.51   478.5  979.72   486.4  984.68   502.3 1000.46
   506.3 1003.15   526.2 1012.16   581.8 1034.38   613.6 1044.12   633.4 1048.89
   689.1 1066.73   736.7 1083.13   744.7 1087.42   764.6 1087.46   820.2 1102.05
#Mann= 3 , 0 , 0
       0     .08       0   403.4    .045       0   418.4      .1       0
Bank Sta=403.4,418.4
XS Rating Curve= 0 ,0
Exp/Cntr=0.3,0.1

Type RM Length L Ch R = 1 ,31909.7 ,250.5,248.2,243.5
XS GIS Cut Line= 3
     1751455.713      337685.183     1751864.091      337714.435
     1752271.403      337760.688
#Sta/Elev= 30
       0 1064.23    15.9 1051.86    27.8 1046.88    67.6  1013.9   111.3   974.4
   119.2  969.85   143.1  969.29     159  966.89   206.7     966   274.3  967.58
     326  964.83   369.7  965.46   381.6  964.47   393.5  959.44   401.9  958.81
   413.4  958.68   416.9  958.86   441.3  964.06     493  966.01   512.9  976.32
   556.7  976.08   560.7  978.06   576.6  991.62   664.1 1044.32   715.9 1077.73
   723.8 1081.28   735.8 1083.16   751.7 1088.48   787.5 1107.77   819.4 1128.48
#Mann= 3 , 0 , 0
       0     .08       0   401.9    .045       0   416.9      .1       0
Bank Sta=401.9,416.9
XS Rating Curve= 0 ,0
Exp/Cntr=0.3,0.1

Type RM Length L Ch R = 1 ,31661.5 ,377.5,376.8,377.4
XS GIS Cut Line= 3
     1751526.174      337970.831     1751849.091       337962.15
     1752239.716      337927.428
#Sta/Elev= 30
       0 1031.77      16  1019.6    67.8  973.06    75.8  968.88   103.7  969.33
   123.6  966.81   147.6  966.99   179.5  962.63   239.3  964.94   287.1  963.71
   295.1     963     318  957.07     323  956.84     333   957.2   354.7  959.17
   366.6  961.95   386.4  963.12   449.8  963.16   453.8  964.13   469.6  973.08
   505.2  975.35   513.2   980.1   521.1  990.24     529  998.49   552.8 1015.99
   600.3 1046.48   647.9 1075.15   667.7 1080.26   691.4 1090.63   715.2 1103.56
#Mann= 3 , 0 , 0
       0     .08       0     318    .045       0     333      .1       0
Bank Sta=318,333
XS Rating Curve= 0 ,0
Exp/Cntr=0.3,0.1

Type RM Length L Ch R = 1 ,31284.7 ,236.1,238.5,241.3
XS GIS Cut Line= 3
     1751553.897      338322.274     1751970.618      338302.428
     1752376.867      338283.553
#Sta/Elev= 30
       0 1035.64    23.8 1016.73    55.6  994.48    79.5  972.44    87.4  967.34
     155  963.91   266.2  965.59   305.9  963.86   325.8  960.87   353.6  959.31
   377.5  960.85   397.3  955.58   404.2  955.71   419.2  955.66   433.1  957.31
   445.1  967.65   453.1  971.57     485  973.09     493  974.87   496.9  978.29
   508.9  993.97   520.9 1004.67   556.7 1032.56   608.6 1068.57   628.5 1074.65
   664.4 1094.54     776 1171.19     800  1184.8   815.9 1196.06   823.9 1197.54
#Mann= 3 , 0 , 0
       0      .1       0   404.2    .045       0   419.2      .1       0
Bank Sta=404.2,419.2
XS Rating Curve= 0 ,0
Exp/Cntr=0.3,0.1

Type RM Length L Ch R = 1 ,31046.1 ,131.2,151.1,170.4
XS GIS Cut Line= 3
     1751569.577      338514.234     1751965.988      338539.935
     1752370.061      338571.503
#Sta/Elev= 30
       0 1020.93    19.9 1005.94    63.6  967.25    67.5  965.43   202.6  962.52
   365.5  961.61   373.4  960.42   381.4  956.24   389.3  954.53   390.9  954.57
   405.9  955.15   421.1  956.62     437  968.78     441  970.42   472.7  972.07
   480.7  974.72   492.6   983.1   504.5  996.99   512.5  1004.9   532.4 1018.74
   568.1 1037.95   599.9 1052.72   615.8  1062.1   631.7 1066.56   639.6 1072.27
   683.3 1094.55   758.8  1142.4   778.7 1153.86   798.6 1166.65   802.6  1170.3
#Mann= 3 , 0 , 0
       0      .1       0   390.9    .045       0   405.9      .1       0
Bank Sta=390.9,405.9
XS Rating Curve= 0 ,0
Exp/Cntr=0.3,0.1

Type RM Length L Ch R = 1 ,30895   ,90.6,87.4,84.5
XS GIS Cut Line= 6
     1751550.479      338630.553     1751725.827      338595.831
     1751829.993      338599.303     1751918.535      338654.859
     1752015.757      338753.817     1752368.188      338757.289
#Sta/Elev= 30
       0 1030.72    23.8 1012.94    55.6  984.99    83.4  964.47   103.3  965.17
   154.9  962.18     283  960.37   333.3  962.35   348.8  959.49     372  959.95
     430  954.67   431.1   954.6     445  954.87   466.8  955.63   482.6  960.99
   490.6  966.79   498.5  969.39   549.2  971.27   560.6  970.42   564.5  971.79
   572.1  976.97   583.6  990.39     595  999.27   685.5 1061.32   693.4 1068.22
   709.2 1072.28   732.9 1085.51   799.9 1132.97   807.8 1136.97   878.8 1183.14
#Mann= 3 , 0 , 0
       0      .1       0     430    .045       0     445      .1       0
Bank Sta=430,445
XS Rating Curve= 0 ,0
Exp/Cntr=0.3,0.1

Type RM Length L Ch R = 1 ,30807.6 ,413,398,384.6
XS GIS Cut Line= 6
     1751566.104      338705.206     1751680.688      338658.331
     1751784.854      338661.803     1751873.396      338717.359
     1751970.618      338816.317     1752323.049      338819.789
#Sta/Elev= 30
       0 1016.66      12 1009.79    63.9  967.16    71.9  964.28    95.8  964.69
   139.2  959.65   293.8  958.74   317.1  956.57   401.7   953.3   411.8  953.05
   416.7  953.07   423.7   953.2   435.6  958.86   494.2  958.14   509.5  966.19
   517.2  968.54   540.1  970.92   551.7  970.06   559.6  972.42   571.4  983.96
   595.1 1001.87     603 1006.51   614.8  1016.5   681.9 1060.13   693.7    1070
   705.5 1072.08   737.1 1089.84   764.7 1110.37   784.4 1123.16   823.9 1146.02
#Mann= 3 , 0 , 0
       0      .1       0   401.7    .045       0   416.7      .1       0
Bank Sta=401.7,416.7
XS Rating Curve= 0 ,0
Exp/Cntr=0.3,0.1

Type RM Length L Ch R = 1 ,30409.7 ,190.4,192.5,192.6
XS GIS Cut Line= 3
     1751441.104      338969.095     1751650.668      338998.931
     1752165.063       339109.72
#Sta/Elev= 30
       0 1084.42      24 1065.59    43.9 1060.36    55.9 1047.25    91.9 1020.21
   127.8  988.39   131.8  984.27   143.8  966.17   147.8   962.1   151.8  960.46
   175.7  960.37   187.7  952.44   204.2  951.75   219.2  951.34   227.6  950.97
   235.6  952.16   255.5  958.57     419  956.73   554.5  959.39   562.5  960.86
   570.4  965.59   578.4  967.76   598.4  969.32   610.3   967.9   622.3  968.97
   634.2  975.82   654.2  991.75     686 1013.65     702 1026.72   737.9 1048.92
#Mann= 3 , 0 , 0
       0      .1       0   204.2    .045       0   219.2     .06       0
Bank Sta=204.2,219.2
XS Rating Curve= 0 ,0
Exp/Cntr=0.3,0.1

Type RM Length L Ch R = 1 ,30217.2 ,283.9,294.5,304.8
XS GIS Cut Line= 4
     1751413.327      339085.414      1751500.67      339159.597
     1751609.507      339186.109     1752114.716      339298.956
#Sta/Elev= 30
       0 1069.62    15.8 1061.74    27.7 1057.87    47.4 1044.03    59.3 1040.97
    90.9 1021.79   137.8  986.87   149.4  974.84     161  960.46   164.8  958.89
     188  958.88   195.7  955.27   222.8  949.62   223.9  949.67   238.9  949.93
   254.5  950.16   286.3  957.45     358  954.99   497.4   958.8   565.1  958.68
     585  965.52   604.9  967.92   620.8  966.99   632.8  972.28   664.6  995.65
   680.6 1010.26   684.5 1012.51   716.4 1023.48   728.3 1029.44   744.3 1032.95
#Mann= 3 , 0 , 0
       0      .1       0   223.9    .045       0   238.9     .06       0
Bank Sta=223.9,238.9
XS Rating Curve= 0 ,0
Exp/Cntr=0.3,0.1

Type RM Length L Ch R = 1 ,29922.7 ,383.8,413,443.4
XS GIS Cut Line= 4
     1751347.354       339203.47     1751382.094      339342.338
     1751536.591      339470.831     1751897.702      339759.025
#Sta/Elev= 30
       0 1046.16    19.9 1038.89    43.7 1027.63    59.6 1023.86    87.5 1006.78
   119.3  985.01   147.1  960.67     155  955.66   162.8  954.89   186.5  956.29
     281  954.54   308.6     953   334.6  948.27   336.2  948.22   349.6  948.54
     372  949.42   411.8  954.77   551.2  956.28   559.2  957.63   575.1  963.48
     587  965.08     603  964.49     607  966.16   638.8  986.82   686.6 1007.21
   694.6 1009.51   730.4 1015.21   786.2 1035.28   798.1 1037.08   806.1 1040.29
#Mann= 3 , 0 , 0
       0      .1       0   334.6    .045       0   349.6     .06       0
Bank Sta=334.6,349.6
XS Rating Curve= 0 ,0
Exp/Cntr=0.3,0.1

Type RM Length L Ch R = 1 ,29509.7 ,303.4,300,299.5
XS GIS Cut Line= 3
     1751302.216      339309.372     1751187.882      339570.596
     1751025.152      339918.507
#Sta/Elev= 30
       0 1005.39    43.6  979.25    59.4  967.15    67.3  958.88    75.2   953.7
   130.7  954.54   162.4  952.68   170.3   951.1     202  953.11   225.7  949.07
   257.4  948.96   269.3   947.2   277.6  947.38   292.6  946.46     297  946.31
   320.8     948   328.7  950.42   336.6  951.16   443.5  953.92   459.4  956.36
   467.3  959.27     491  961.06   518.8   957.1   526.7  960.92   566.3  993.75
   574.2  998.66   609.8 1011.17   637.6 1018.83   649.4 1023.62   669.2 1024.11
#Mann= 3 , 0 , 0
       0      .1       0   277.6    .045       0   292.6      .1       0
Bank Sta=277.6,292.6
XS Rating Curve= 0 ,0
Exp/Cntr=0.3,0.1

Type RM Length L Ch R = 1 ,29209.7 ,289.3,300,309.1
XS GIS Cut Line= 3
     1751033.273      339002.267      1750913.82      339448.588
     1750751.987       339814.64
#Sta/Elev= 30
       0 1020.45    23.9 1018.44    43.8 1009.62   147.4  978.17   163.3     971
   179.2  967.27   203.1  956.38   215.1  953.02   266.9  952.52   342.5  948.38
   374.4  951.72   386.4  947.69   406.3  948.96   454.5  944.68     462  944.42
   469.5  944.62   485.8  944.96   501.7  948.48   537.3  946.93     577  952.52
   612.6  951.15   632.4  957.27   652.2  959.21     672  955.46   731.5 1004.46
   775.1 1024.84     783 1030.82   798.9  1034.9   810.7 1044.74   862.3 1078.96
#Mann= 3 , 0 , 0
       0      .1       0   454.5    .045       0   469.5      .1       0
Bank Sta=454.5,469.5
XS Rating Curve= 0 ,0
Exp/Cntr=0.3,0.1

Type RM Length L Ch R = 1 ,28909.7 ,295.4,300,302.8
XS GIS Cut Line= 3
     1750962.099      338955.468     1750680.195      339267.573
     1750383.347      339546.813
#Sta/Elev= 30
       0 1001.88    19.8  991.68    51.6   980.9    87.3  963.15   107.1  958.29
   150.8  955.92   174.6   958.2   210.3  950.58   317.4   950.3   333.3  947.17
   353.1   949.5     369  945.82   413.1     943   424.6  942.23   428.1  942.37
   476.5  946.64   496.5  955.89   528.4  957.05   532.4  958.97   560.4  984.94
   580.4  999.83   624.3 1022.39   636.3 1024.97   684.3 1059.28   704.2  1077.3
   744.2 1106.18   780.2 1127.18   792.2 1131.38   796.2 1135.71   828.1 1156.03
#Mann= 3 , 0 , 0
       0      .1       0   413.1    .045       0   428.1      .1       0
Bank Sta=413.1,428.1
XS Rating Curve= 0 ,0
Exp/Cntr=0.3,0.1

Type RM Length L Ch R = 1 ,28609.7 ,299.9,300,300.1
XS GIS Cut Line= 3
     1750838.075      338781.694      1750507.41      339023.065
     1750176.516      339264.577
#Sta/Elev= 30
       0 1000.81    59.6  964.75    79.5  956.52    95.4  957.28   119.2  951.92
   230.5  952.06   254.4  954.87   274.2  948.84     318  949.52   361.7  945.29
   381.6  945.59   397.5  939.37   401.9  939.55   416.9  939.65   449.2  944.74
     469   954.1   504.8  954.92   516.8   969.9   532.7   978.9   540.6  989.44
   548.6  996.31   592.3 1019.21   608.2 1024.04     652 1054.86     660 1058.27
   691.8  1083.4   723.6  1104.4   743.5 1117.03   755.4 1119.84     819 1159.24
#Mann= 3 , 0 , 0
       0      .1       0   401.9    .045       0   416.9      .1       0
Bank Sta=401.9,416.9
XS Rating Curve= 0 ,0
Exp/Cntr=0.3,0.1

Type RM Length L Ch R = 1 ,28309.7 ,304.3,300,295.2
XS GIS Cut Line= 3
     1750656.067      338545.379     1750324.324      338785.455
     1749992.582      339025.532
#Sta/Elev= 30
       0  1011.6    51.7  982.75    71.6  966.38    83.5   963.6    95.4  956.16
   135.2  951.95   258.4  952.25   286.2  955.84   306.1  947.16   345.9  947.84
   361.8  943.03   377.7  943.18   397.6   938.3     402  938.34     417  938.41
   445.3  943.28   461.2  951.68     497  953.93   508.9  966.94   524.8  975.07
   536.7  992.39   560.6 1010.47   584.4 1024.65   600.3 1028.75   667.9 1076.84
   731.5 1109.57   747.4 1114.77   767.3 1126.94   795.2 1139.79     819 1155.02
#Mann= 3 , 0 , 0
       0      .1       0     402    .045       0     417      .1       0
Bank Sta=402,417
XS Rating Curve= 0 ,0
Exp/Cntr=0.3,0.1

Type RM Length L Ch R = 1 ,28009.7 ,306.9,300,293.5
XS GIS Cut Line= 3
     1750405.865      338261.913     1750126.326       338561.14
     1749852.186      338865.449
#Sta/Elev= 30
       0 1042.06    15.9 1038.21    39.8 1022.55    55.7 1018.38   143.1  970.52
     171  957.14   182.9  953.18   238.5  949.83   302.1  949.53     334  944.35
   361.8  944.98   385.6  938.05   397.6  937.22     402  937.26     417  937.41
   457.2  942.86   481.1  941.87     489  943.82     501  950.29   532.8  952.87
   552.6  972.74   556.6  975.93   572.5  982.35   588.4  999.16   604.3 1010.39
   648.1 1035.37     664 1039.37   775.3 1108.78   787.2 1112.77   819.1 1131.24
#Mann= 3 , 0 , 0
       0      .1       0     402    .045       0     417      .1       0
Bank Sta=402,417
XS Rating Curve= 0 ,0
Exp/Cntr=0.3,0.1

Type RM Length L Ch R = 1 ,27709.7 ,305.5,300,294.5
XS GIS Cut Line= 3
     1750046.205      338039.611     1749870.013      338409.268
     1749693.821      338778.926
#Sta/Elev= 30
       0 1058.19    35.8 1035.15    47.7 1032.55    75.5 1017.24   123.2  973.81
   139.2  972.24     159  954.14     171  947.04   186.9  948.88   202.8  945.36
   290.2  944.58     326   947.7   341.9  943.16   369.7  942.35     402  936.01
   405.5     936     417  936.21   445.3  940.54   500.9   940.5   520.8  948.62
   540.7  950.44   552.6  948.71   560.6  950.96   576.5  971.27   588.4  982.14
   632.1  1014.2   667.9 1036.21   687.8 1042.63   779.2 1105.41     819 1121.11
#Mann= 3 , 0 , 0
       0     .08       0     402    .045       0     417      .1       0
Bank Sta=402,417
XS Rating Curve= 0 ,0
Exp/Cntr=0.3,0.1

Type RM Length L Ch R = 1 ,27409.7 ,309.3,300,291.2
XS GIS Cut Line= 3
     1749672.327       337901.85     1749591.098      338303.212
     1749509.869      338704.575
#Sta/Elev= 30
       0 1019.28    51.7   993.6    71.6  980.95   127.2  957.86     155  944.54
     159  944.16     171  947.69   210.7  947.52   238.5  941.45   381.7  940.72
     402  935.13   409.5  934.54     417  934.89   433.4   935.3   457.2   940.6
     493  939.74   540.7  948.72   556.6  947.22   572.5  948.07   580.5  953.22
   596.4  970.06   616.2  987.92     652 1015.96   683.8 1036.94   695.8 1042.75
   707.7 1043.95   711.7 1046.18   795.2 1112.55   807.1 1116.39     819 1124.66
#Mann= 3 , 0 , 0
       0     .08       0     402    .045       0     417      .1       0
Bank Sta=402,417
XS Rating Curve= 0 ,0
Exp/Cntr=0.3,0.1

Type RM Length L Ch R = 1 ,27109.7 ,302.8,300,297.3
XS GIS Cut Line= 3
     1749196.313       337828.47     1749294.748      338284.615
     1749356.035      338595.831
#Sta/Elev= 30
       0  980.17    23.9  973.17    43.9  970.96    67.8  965.37    87.8  964.25
    99.7  968.35   111.7  967.48   131.6  960.02   147.6  948.93   155.6  947.02
   259.2  942.34   291.2  943.13   390.9  940.34   434.7   941.6   442.7  940.25
   450.7  933.57   454.7  932.97   459.1     933   474.1  933.27   502.3  936.73
   545.9   937.5   561.8   945.7   597.5   946.2   609.4  948.69   633.2  966.75
     653  992.43   676.8  1015.2   716.4 1039.49   732.3 1043.76   783.8 1079.34
#Mann= 3 , 0 , 0
       0     .08       0   459.1    .045       0   474.1      .1       0
Bank Sta=459.1,474.1
XS Rating Curve= 0 ,0
Exp/Cntr=0.3,0.1

Type RM Length L Ch R = 1 ,26809.7 ,332.9,308.9,284.9
XS GIS Cut Line= 5
     1749081.729      337786.803     1748933.863      338156.091
     1749022.116      338408.132     1749067.841      338554.164
     1749294.087        338746.3
#Sta/Elev= 30
       0  995.73    59.7  967.89    71.6   958.3    79.6  955.09    99.4  959.16
   119.3  960.34   159.1  954.96     362   951.3   509.4  943.61   533.3  935.16
     633  936.17   656.9   932.2   657.3  932.21   672.3  932.52   688.4  932.87
   700.2  936.45   735.5  936.63   755.1  943.64   821.8  945.71   829.7  949.15
   845.6  968.03   865.4  981.04   885.1 1002.97   893.1 1009.14   956.4 1025.22
  1003.9 1040.37  1019.7  1042.5  1043.4 1051.13  1067.2 1054.32  1114.7 1072.41
#Mann= 3 , 0 , 0
       0      .1       0   657.3    .045       0   672.3      .1       0
Bank Sta=657.3,672.3
XS Rating Curve= 0 ,0
Exp/Cntr=0.3,0.1

Type RM Length L Ch R = 1 ,26500.7 ,289.6,291.1,292.3
XS GIS Cut Line= 3
     1748433.787      338545.428     1748823.049        338618.4
     1749079.993      338677.428
#Sta/Elev= 30
       0 1026.19    23.8 1007.51    35.6  1002.3    67.3  982.35    83.2  970.28
   114.8  941.77   122.8  937.24   126.7  935.78   166.3  934.48   178.2  929.38
   186.1  929.12   225.7  934.54   265.4  930.33   368.3  935.41   380.2  931.47
   394.1  930.66   409.1  931.14     428  933.76   471.9  932.77   531.9   934.8
   539.8  936.85   547.8  943.01   551.8  943.97   591.8  944.53   599.8  947.02
   611.8  958.66   627.7  970.14   639.7  983.29   643.7  986.25   659.7  992.69
#Mann= 3 , 0 , 0
       0      .1       0   394.1    .045       0   409.1      .1       0
Bank Sta=394.1,409.1
XS Rating Curve= 0 ,0
Exp/Cntr=0.3,0.1

Type RM Length L Ch R = 1 ,26209.7 ,250.5,244.3,237.7
XS GIS Cut Line= 3
     1748399.682      338799.188     1748810.874      338907.654
     1749201.944      339019.389
#Sta/Elev= 30
       0  1078.3    43.7 1049.63    55.6 1038.77    95.4 1018.08   119.2  999.15
   131.2  994.64   186.8  960.29   214.6  934.88   222.6  932.45   266.3  931.52
   290.1   926.8   298.1  926.97     310  931.87   349.7  933.13   365.6  930.56
   393.5  932.02   417.8  928.77   432.8  929.32   453.2  933.15   556.8  931.77
   576.8  940.53   592.7     943   616.6  941.99   628.6  938.49   652.5  940.47
   664.5   944.2   688.4   958.6   712.4  966.01   772.2  992.15     832 1024.88
#Mann= 3 , 0 , 0
       0      .1       0   417.8    .045       0   432.8      .1       0
Bank Sta=417.8,432.8
XS Rating Curve= 0 ,0
Exp/Cntr=0.3,0.1

Type RM Length L Ch R = 1 ,25965.3 ,351.3,355.7,356.7
XS GIS Cut Line= 3
     1748451.521      339135.761     1748797.842      339132.771
     1749192.023      339106.939
#Sta/Elev= 30
       0 1109.64    31.8 1091.91    55.7 1074.73    67.7 1064.93    87.6 1044.74
   107.5 1029.38   135.4 1012.54   143.3 1006.06   159.2 1000.46   175.2  989.05
     207  961.54   226.9  937.96   230.9  934.84   254.8  934.33   270.7  927.32
     285  926.34   294.6  926.28     300   926.5   318.5  929.61   358.3   931.4
     486  931.86     498  933.71   509.9  939.59   525.9  941.97   565.8  937.16
   601.7  939.35   621.7   947.4   661.6  971.58   709.4  996.95   741.4 1016.71
#Mann= 3 , 0 , 0
       0      .1       0     285    .045       0     300      .1       0
Bank Sta=285,300
XS Rating Curve= 0 ,0
Exp/Cntr=0.3,0.1

Type RM Length L Ch R = 1 ,25609.7 ,294.6,300,308
XS GIS Cut Line= 4
      1748434.16      339357.984     1748661.661      339427.498
     1748914.117      339438.117     1749302.216      339434.372
#Sta/Elev= 30
       0  1060.1    27.8 1046.03    51.5  1031.5    63.4 1029.61    87.2  1017.6
   103.1 1012.93   182.4  976.35     222  954.81   245.8  935.27   269.5  936.86
   285.3  929.37   427.4  927.33   451.1  928.47   483.1   924.8   490.6  924.65
   498.1  924.88   518.3  925.87   538.1  937.09     542  937.87   561.8  939.81
   585.6  935.91   593.5  937.76   621.3  952.07   637.1  962.83   680.7  995.51
   696.5 1009.21   759.9 1037.33   779.7  1051.7   835.1 1087.09   878.7 1108.09
#Mann= 3 , 0 , 0
       0      .1       0   483.1    .045       0   498.1      .1       0
Bank Sta=483.1,498.1
XS Rating Curve= 0 ,0
Exp/Cntr=0.3,0.1

Type RM Length L Ch R = 1 ,25309.7 ,300.7,300,301.6
XS GIS Cut Line= 3
     1748377.616      339488.358     1748816.313      339692.511
     1749112.979      339831.942
#Sta/Elev= 30
       0 1029.74     164  971.83     204  955.62   227.9  939.32   251.9  939.55
   263.9  934.88   275.9  933.11   351.9  930.06   403.9  924.68   447.9  925.59
   476.4  923.85   487.9  922.92   491.4  923.02   503.9  923.41   519.8  927.49
   567.8  928.52   575.8  931.03   583.8  936.02   619.8   936.8   643.8  940.07
   659.8  966.31   667.8  977.42   671.8  981.05   683.8  986.73   707.7 1003.54
   723.7 1009.07   751.7 1029.11   779.7 1052.01   799.7 1063.76   811.7 1072.84
#Mann= 3 , 0 , 0
       0      .1       0   476.4    .045       0   491.4      .1       0
Bank Sta=476.4,491.4
XS Rating Curve= 0 ,0
Exp/Cntr=0.3,0.1

Type RM Length L Ch R = 1 ,25009.7 ,277.1,300,321.2
XS GIS Cut Line= 5
     1748336.159      339552.854     1748472.354      339851.039
     1748683.788      339937.761     1748798.743      339995.136
     1749019.229      339967.359
#Sta/Elev= 30
       0 1014.14      16 1009.76      56  990.92      68  988.69   103.9  974.35
   207.9  945.24   223.9  936.86   247.9  938.66   263.8  931.14   303.8  928.96
   351.5  930.06   398.7  927.26   516.9  929.21   532.7  921.95   540.6  921.31
   548.8   921.4   563.8   921.8   587.5  925.09   630.3  925.72   649.8  933.36
     677  935.29   696.7  945.82   720.5  942.51   776.1  940.79     784  944.34
   795.9  955.16   811.8   965.1   859.4  984.33   891.2 1004.53     907 1009.77
#Mann= 3 , 0 , 0
       0      .1       0   548.8    .045       0   563.8      .1       0
Bank Sta=548.8,563.8
XS Rating Curve= 0 ,0
Exp/Cntr=0.3,0.1

Type RM Length L Ch R = 1 ,24709.7 ,293.8,300,306.2
XS GIS Cut Line= 3
     1748352.563      339613.192     1748452.648       340075.15
     1748528.337      340458.328
#Sta/Elev= 30
       0     989     7.9  987.67    23.8  980.42    75.5  962.63   150.9  942.08
   166.8  935.68   182.7  937.59   202.6  936.94   250.2  927.72   373.4  926.87
   393.2  923.57   448.8  922.56   464.7  919.43   465.2  919.44   480.2  919.74
   496.6  920.74   508.6  928.65   516.5  931.41   544.4  933.47   548.4   937.1
   560.4  958.29   564.3  963.42   568.3  966.04   636.1 1003.58   679.9 1034.72
   699.8 1045.84   743.7 1068.06   783.6 1082.52   795.5 1091.62   863.3 1134.31
#Mann= 3 , 0 , 0
       0      .1       0   465.2    .045       0   480.2      .1       0
Bank Sta=465.2,480.2
XS Rating Curve= 0 ,0
Exp/Cntr=0.3,0.1

Type RM Length L Ch R = 1 ,24409.7 ,290,300,312.9
XS GIS Cut Line= 3
     1748191.931      339596.102     1748156.896      340076.772
     1748128.604       340462.15
#Sta/Elev= 30
       0 1006.22    55.8   982.9   143.4  949.73   155.3  944.45   167.3  934.89
   195.2  935.44   207.1  930.02     231  927.19   354.5  926.23   398.3  920.28
   450.1  921.76     470  917.47   474.4  917.47   489.4  917.49   505.8  919.06
   521.8  928.54   549.7  931.16   553.6  933.67   565.6  953.17   573.6  959.75
   637.3 1002.89   669.2 1028.18   740.9 1079.86   752.8 1085.42   764.8 1095.03
   816.6 1129.77   828.5 1139.69   840.5 1145.48   848.4 1152.67   868.4 1165.63
#Mann= 3 , 0 , 0
       0      .1       0   474.4    .045       0   489.4      .1       0
Bank Sta=474.4,489.4
XS Rating Curve= 0 ,0
Exp/Cntr=0.3,0.1

Type RM Length L Ch R = 1 ,24109.7 ,296.1,300,300.5
XS GIS Cut Line= 3
     1748116.556      339562.635     1747908.839      339922.551
     1747654.968      340252.013
#Sta/Elev= 30
       0  1018.1    79.9  979.18    95.9  973.93   123.9  959.28   135.8  951.78
   147.8  939.73   155.8  934.46   179.8  934.39   195.8  926.75   255.7     926
   275.7  920.47   387.6  920.52   407.6  915.81   408.1  915.82   423.1  916.03
   451.6  917.38   459.6  919.92   471.6  926.92   487.5  929.58   507.5  929.37
   539.5  951.42   559.5  957.46   579.5  966.42   591.5  973.96   607.5  979.34
   615.5  985.25   775.5 1079.23   787.5 1081.87   799.5 1090.61   831.5 1109.28
#Mann= 3 , 0 , 0
       0      .1       0   408.1    .045       0   423.1      .1       0
Bank Sta=408.1,423.1
XS Rating Curve= 0 ,0
Exp/Cntr=0.3,0.1

Type RM Length L Ch R = 1 ,23809.7 ,301.5,300,298.5
XS GIS Cut Line= 3
     1747918.349      339444.798     1747660.416      339762.856
     1747402.484      340080.914
#Sta/Elev= 30
       0  1041.7    47.7 1005.82    63.6  997.81    79.5     987   107.3  975.81
   147.1  955.98     171  933.94   198.8  933.31   214.7  923.77   222.6  922.59
   341.9  923.15   349.9  922.32   361.8  917.92     402  914.48   413.5  914.17
     417  914.31   433.4  914.99   457.2  926.19     489  928.65   516.8  943.63
   548.6  950.27   572.5   957.3   588.4  964.17   604.3  966.27   636.1   976.8
   683.8    1004   699.7 1010.88   715.6 1023.93   751.4 1047.27     819 1085.83
#Mann= 3 , 0 , 0
       0      .1       0     402    .045       0     417      .1       0
Bank Sta=402,417
XS Rating Curve= 0 ,0
Exp/Cntr=0.3,0.1

Type RM Length L Ch R = 1 ,23509.7 ,276.5,277.4,276.6
XS GIS Cut Line= 3
     1747653.115      339251.962     1747417.557      339586.929
     1747181.999      339921.896
#Sta/Elev= 30
       0 1052.53    59.6 1007.77    99.4  985.99   139.2  971.12   182.9  951.76
   190.8  946.83   206.7  932.74   210.7  930.96   242.5  930.22   254.4  923.85
   266.4  920.52     326  919.26   365.8  920.67     402  913.17   409.5  913.02
     417  913.14   469.1   923.5     489  926.02   512.9  923.24   528.8  924.94
   540.7  928.97   568.5   942.9   588.4  950.58   612.3  955.53   667.9  972.85
   687.8  977.21   731.5  995.92   751.4 1006.56   779.2 1025.07     819  1048.9
#Mann= 3 , 0 , 0
       0      .1       0     402    .045       0     417      .1       0
#XS Ineff= 2 , 0
                          492.93          934.48
Permanent Ineff=
       F       F
Bank Sta=402,417
XS Rating Curve= 0 ,0
Exp/Cntr=0.3,0.1

Type RM Length L Ch R = 1 ,23232.2 ,335.7,322.6,310.8
XS GIS Cut Line= 4
     1747459.263      339092.931     1747206.729      339406.595
      1747061.08      339630.146     1747052.216      339779.859
#Sta/Elev= 30
       0 1073.12    43.9 1044.92    87.7 1012.42   127.6  988.41   159.5  975.36
   187.4  968.79   215.3  957.11   239.2   946.9   251.2  936.04   255.2  934.18
   287.1  932.01     311  918.04   362.8  918.08   386.7  914.84   400.2  911.23
   410.6  910.86   415.2  910.92   446.5  916.74   458.4  916.85   470.4  919.79
   542.1  920.73   569.9  924.54   601.8  920.82   661.5  922.14   681.3  928.08
     709  941.51   736.6  952.83   776.1  961.63   795.8  968.53   819.5  973.76
#Mann= 3 , 0 , 0
       0      .1       0   400.2    .045       0   415.2      .1       0
#XS Ineff= 2 , 0
                          569.81          933.86
Permanent Ineff=
       F       F
Bank Sta=400.2,415.2
XS Rating Curve= 0 ,0
Exp/Cntr=0.3,0.1

Type RM Length L Ch R = 1 ,22909.7 ,309.1,300,289.3
XS GIS Cut Line= 3
     1746942.841      339031.595     1746924.446      339268.282
        1746897.      339731.226
#Sta/Elev= 30
       0 1016.01    15.8 1002.94    51.4  988.12      91   977.7   138.5  956.12
   150.4  946.51   154.3  945.39     186  944.03   189.9   941.9   205.8  927.26
   217.6  912.98   221.6  910.76   229.9  909.87   244.9  909.56   253.4  909.77
   273.4  913.79   289.4  913.96   333.4   918.3   473.3  917.16   481.3  918.14
   489.3  921.32   505.3  923.57   521.2  920.67   529.2  916.79   541.2   916.4
   633.2  931.55   673.2  941.61   685.2  945.96   693.2  947.12   701.2  950.79
#Mann= 3 , 0 , 0
       0      .1       0   229.9    .045       0   244.9      .1       0
#XS Ineff= 2 , 0
                          501.07          932.29
Permanent Ineff=
       F       F
Bank Sta=229.9,244.9
XS Rating Curve= 0 ,0
Exp/Cntr=0.3,0.1

Type RM Length L Ch R = 1 ,22609.7 ,312.7,300,289.4
XS GIS Cut Line= 3
     1746507.658      338962.997     1746635.987      339345.947
     1746813.287      339750.114
#Sta/Elev= 30
       0 1102.59      56  1073.6      84 1049.86     100  1040.8     148 1000.61
     164  989.49     180  982.87   195.9  980.33   215.9  973.36   247.9  953.84
   275.9  951.43   291.9  943.12   331.9  937.05   347.9  929.08   371.9  911.55
   396.4  908.92   403.9  908.78   411.4  909.05   423.8  909.34   439.7  913.19
   467.5  911.84   487.4  914.71     551  914.75   634.5  926.37   646.4  923.15
   670.3  922.53   690.2   931.8   789.6  938.21   825.4  943.87   845.2  949.17
#Mann= 3 , 0 , 0
       0      .1       0   396.4    .045       0   411.4      .1       0
Bank Sta=396.4,411.4
XS Rating Curve= 0 ,0
Exp/Cntr=0.3,0.1

Type RM Length L Ch R = 1 ,22309.7 ,230.3,232,233.7
XS GIS Cut Line= 3
     1746078.368      339251.116     1746387.665      339504.949
     1746743.624      339798.517
#Sta/Elev= 30
       0 1108.79    19.8 1096.67    63.4 1065.52    79.2  1050.7    95.1  1039.8
   142.6 1001.56   186.2  975.08     206  955.34     210   952.7   229.8  951.34
   237.7  948.16   269.4  921.82   281.3   914.8   301.1  908.05   372.4  910.31
   392.2  906.17   392.6  906.18   407.6  906.22     428  906.68   451.8  910.37
   487.6  908.94   507.5  911.58   563.2  913.47   618.9  920.61   662.6  922.79
   674.6  921.73   686.5  925.42   742.2  934.44   825.7  943.98   861.5  951.67
#Mann= 3 , 0 , 0
       0      .1       0   392.6    .045       0   407.6      .1       0
Bank Sta=392.6,407.6
XS Rating Curve= 0 ,0
Exp/Cntr=0.3,0.1

Type RM Length L Ch R = 1 ,22077.6 ,382.1,368,354.4
XS GIS Cut Line= 4
     1746001.961      339411.048      1746307.62      339705.643
     1746504.574      339889.934     1746649.438      339958.678
#Sta/Elev= 30
       0 1079.12    31.7 1059.08    47.6 1040.79    67.4    1025    83.3 1010.12
     123  980.24   146.8  957.39   150.8  955.67   174.6  954.01   214.2  932.55
     242  910.25   257.9   906.9   297.6  907.88   321.4  912.04   357.1  911.68
   376.9  910.13   392.8  906.48   408.6  908.92   441.2   905.9   460.2  904.89
   468.2   905.9     488  911.36   567.3  909.87   591.1  911.03     611  918.83
   626.8  920.85   642.7   920.1   729.4  935.14   752.9  936.24   854.6  960.54
#Mann= 3 , 0 , 0
       0      .1       0   441.2    .045       0   468.2      .1       0
Bank Sta=441.2,468.2
XS Rating Curve= 0 ,0
Exp/Cntr=0.3,0.1

Type RM Length L Ch R = 1 ,21709.7 ,242,238.3,233.8
XS GIS Cut Line= 3
      1745934.16      339951.734     1746117.327       339973.77
     1746552.216      340036.803
#Sta/Elev= 30
       0 1007.98     7.8  998.49    23.6  984.54    39.2  966.75      51  956.08
    62.8  952.78    78.5  951.12    82.4  949.19   121.7  917.67   141.3   904.5
   145.2  903.71     157  904.67     177  902.56   184.5  902.35     192  902.35
   204.5  903.25   212.4  906.29   276.4   907.5   344.3  911.28   408.2   910.5
   436.2   911.3   440.2  911.87   452.1  917.37   460.1   919.5   480.1   918.4
   496.1  919.05     548   927.2     564  931.15     584   932.2   623.9  944.63
#Mann= 3 , 0 , 0
       0      .1       0     177    .045       0     192      .1       0
Bank Sta=177,192
XS Rating Curve= 0 ,0
Exp/Cntr=0.3,0.1

Type RM Length L Ch R = 1 ,21471.4 ,249.7,253.2,256.9
XS GIS Cut Line= 4
      1745934.16      340158.331      1746022.59      340214.977
     1746119.924      340210.414     1746533.118      340187.845
#Sta/Elev= 30
       0  993.82    15.6  989.04    38.9  974.51    58.3  964.85    66.1  959.69
    89.5   938.9    97.2   936.5   116.7  935.77   136.2   921.2   159.6  907.46
   175.2  902.05   190.8  901.41   198.6  901.19   205.8  901.46   218.4  901.98
   230.3  904.44   246.2  905.97   262.1  909.34   274.1   907.9   301.9  907.52
   341.7  912.03   389.5  913.99   401.4  916.85   421.3  919.39   441.2  916.26
   461.1  917.19     485  921.65   528.7  925.96   544.6   931.9   616.3  950.61
#Mann= 3 , 0 , 0
       0      .1       0   190.8    .045       0   205.8      .1       0
Bank Sta=190.8,205.8
XS Rating Curve= 0 ,0
Exp/Cntr=0.3,0.1

Type RM Length L Ch R = 1 ,21218.1 ,45.3,45.3,45.3
XS GIS Cut Line= 6
     1745856.035      340361.456     1746010.549      340443.053
     1746195.898      340463.421     1746283.118      340255.553
     1746364.716      340232.984     1746501.868      340260.761
#Sta/Elev= 30
       0  934.15    23.8  929.38   115.2  919.67   178.7  910.97   194.6  909.79
   210.4  910.34   238.2  906.98   250.1  908.11     258  908.11     262  907.48
   277.9  902.79   289.8   901.9   297.7   900.6   309.6   899.5   325.5  899.75
   329.5  900.99   333.4  903.11   345.3  911.72   353.3  913.45   376.4  915.64
   406.9  916.84   536.3  916.45   571.5  917.09     591  916.25   625.6  919.55
   679.7  919.71   711.7  922.12   751.6  926.54   767.6  932.26   815.6  946.19
#Mann= 3 , 0 , 0
       0      .1       0   297.7    .045       0   329.5     .06       0
Bank Sta=297.7,329.5
XS Rating Curve= 0 ,0
Exp/Cntr=0.3,0.1

Type RM Length L Ch R = 1 ,21172.8 ,104.9,115.4,125.3
XS GIS Cut Line= 6
     1745852.563      340406.595     1746007.077      340488.192
     1746210.582      340510.555     1746303.952      340285.067
      1746371.66      340260.761     1746505.858      340293.506
#Sta/Elev= 30
       0  941.53    87.4  930.59   103.2   926.9   115.2  922.91     131   915.6
   178.7  908.17   210.2  908.81   233.8  908.18   241.7  906.98   257.4  902.76
     285  901.77   292.8  900.33   300.7   899.6   313.2  899.93   328.3  901.81
   340.1  906.65   359.8  913.09   395.4   916.4   439.1  918.53   533.2  917.62
   636.3  918.94   648.3   917.9   652.3  918.73   664.3  924.64   668.3  925.55
   727.6  925.74   766.7  927.96   786.2  931.48   805.3  938.66   838.5  949.03
#Mann= 3 , 0 , 0
       0      .1       0   292.8    .045       0   313.2     .06       0
Bank Sta=292.8,313.2
XS Rating Curve= 0 ,0
Exp/Cntr=0.3,0.1

Type RM Length L Ch R = 1 ,21057.4 ,229.8,247.7,266.5
XS GIS Cut Line= 3
     1745842.146      340439.581     1746095.618      340607.984
     1746307.424      340736.456
#Sta/Elev= 30
       0  940.51    35.6  937.11      83  930.61    98.8  926.43   126.5  914.48
   142.3  911.01   197.6  907.14   241.1  908.34   260.8  902.79   272.7  902.54
   292.5  899.35   302.6  898.96   317.6  898.82   320.3  898.77   332.3  899.96
   344.3   903.8   360.2  905.49   364.2  907.07   372.2  912.89   376.2  914.64
   388.2  916.71   400.2  916.63   404.2  918.56   416.2  929.75   420.2  931.52
   432.2  933.45   472.1  944.11   484.1  945.51   536.1  970.67     552  981.44
#Mann= 3 , 0 , 0
       0     .08       0   302.6    .045       0   317.6      .1       0
Bank Sta=302.6,317.6
XS Rating Curve= 0 ,0
Exp/Cntr=0.3,0.1

Type RM Length L Ch R = 1 ,20809.7 ,308,309.6,311.3
XS GIS Cut Line= 3
     1745856.035      340472.567     1745917.972      340764.794
      1745965.41      340995.136
#Sta/Elev= 30
       0  935.65    63.7  922.01    67.7  920.98    79.7  916.01   127.4  911.81
   215.1  905.73     243  907.65   246.9  907.25   254.9  904.14   262.9  903.18
   274.8  898.38   291.2  896.84   306.2   896.7   306.7  896.69   318.6  897.97
   334.6  903.75   346.6  911.34   350.5  912.61   358.5  914.83   370.5  915.12
   374.4  916.66   378.4  923.74   386.4  934.16   394.4  940.52   438.2  961.72
   458.2  976.08   474.1  990.38     498 1008.54     510 1016.71   533.9 1031.52
#Mann= 3 , 0 , 0
       0     .08       0   291.2    .045       0   306.2      .1       0
Bank Sta=291.2,306.2
XS Rating Curve= 0 ,0
Exp/Cntr=0.3,0.1

Type RM Length L Ch R = 1 ,20500.1 ,293,290.4,289.1
XS GIS Cut Line= 5
     1745612.979      340406.595     1745581.094      340542.414
     1745612.979      340785.067     1745641.944      341026.431
      1745715.41      341147.914
#Sta/Elev= 30
       0  950.66    43.8   942.2   127.6  915.16   147.4  910.12   167.1  908.38
   226.4  908.29   317.1  902.87   344.8  903.47   360.6   896.3   372.4  894.96
   374.6  894.96   389.6  895.33   400.2  895.53   420.1  900.36     444  900.71
   467.9  912.26   475.9  913.81   487.9   913.5   495.8  918.56   507.8  932.21
   519.8  939.79   539.7  943.54   559.6  951.75   583.5   958.6   607.4  973.19
     651    1008   686.5 1034.44   725.9 1050.04   737.8 1059.18   769.3 1078.71
#Mann= 3 , 0 , 0
       0     .08       0   374.6    .045       0   389.6      .1       0
Bank Sta=374.6,389.6
XS Rating Curve= 0 ,0
Exp/Cntr=0.3,0.1

Type RM Length L Ch R = 1 ,20209.7 ,250.2,250.7,248.9
XS GIS Cut Line= 5
     1745378.604      340449.997     1745275.418      340617.307
     1745328.066      340821.319     1745373.396      341068.053
      1745573.69      341222.525
#Sta/Elev= 30
       0  940.92    15.7  937.72    62.9  919.08    78.6  916.15   192.6  912.12
   319.8  904.31   363.5  903.75   375.5  901.58   391.4  895.29   399.8  894.38
   414.8  893.97   415.2  893.96   427.2  894.85   443.1   898.1   490.9  898.41
   506.8  903.56   510.8  903.92   550.6  903.92   574.5  905.02   610.4  907.38
   630.3   911.9   642.2   912.6   658.1  911.69     666  915.26   677.9     925
   681.8  926.88   780.6  969.75   843.9 1001.73   895.3 1024.98   911.1 1032.89
#Mann= 3 , 0 , 0
       0      .1       0   399.8    .045       0   414.8      .1       0
Bank Sta=399.8,414.8
XS Rating Curve= 0 ,0
Exp/Cntr=0.3,0.1

Type RM Length L Ch R = 1 ,19959   ,399,364.8,334.8
XS GIS Cut Line= 4
     1745029.646      340644.442     1745088.674      340892.706
     1745159.854      341160.067     1745444.577      341194.789
#Sta/Elev= 30
       0  949.64      12  946.88    43.9  942.54    59.8   937.9    75.8  932.47
    91.7  922.59   103.7  920.98   115.6  914.62   139.6   913.9   147.5  912.27
   171.4  899.02   179.4  897.69   219.3  897.07   259.1  892.83   263.1  892.73
   286.8  893.37   330.3  900.81   413.3  900.96   468.6  902.87   508.1   902.9
   551.8  905.95   607.6  905.43   623.5  906.93   651.4  914.06   671.3  912.04
   691.2  911.67   699.2  915.63   719.1  936.24   774.9  954.33   818.7  970.54
#Mann= 3 , 0 , 0
       0      .1       0   259.1    .045       0   286.8     .08       0
Bank Sta=259.1,286.8
XS Rating Curve= 0 ,0
Exp/Cntr=0.3,0.1

Type RM Length L Ch R = 1 ,19594.2 ,287.1,284.5,280.1
XS GIS Cut Line= 4
     1744639.021      341246.872     1745029.646      341201.734
     1745356.035      341217.359      1745434.16      341224.303
#Sta/Elev= 30
       0 1131.27    51.6 1103.66    71.5  1097.5    99.3 1076.98   127.1  1061.4
     147 1046.57   174.8 1029.14   246.3  973.28     282  941.77     290  938.09
   305.8  937.87   313.8  935.82   345.6  909.05   361.4  893.27   365.4  891.27
   380.3  890.68   389.2  890.53   395.3  890.66   405.2  891.43   417.1  895.71
     465  897.36   488.9  902.61   512.8  905.01   588.5  905.17   608.4  906.52
   636.3  911.92   672.2  911.54   692.1  921.08     712  936.23   798.4  968.03
#Mann= 3 , 0 , 0
       0      .1       0   380.3    .045       0   395.3     .08       0
Bank Sta=380.3,395.3
XS Rating Curve= 0 ,0
Exp/Cntr=0.3,0.1

Type RM Length L Ch R = 1 ,19309.7 ,301.4,300,296.8
XS GIS Cut Line= 3
     1744693.816      341574.364     1745091.631      341478.793
     1745497.507      341410.537
#Sta/Elev= 30
       0 1138.65    63.6 1099.98    79.4 1095.44   150.9 1049.15   190.7 1025.92
   222.4 1002.53     278   959.1   297.9  940.32   305.9  934.18   313.8  931.63
   329.7   931.7   337.6  930.08   357.5  913.92   373.4  903.78   385.3  893.44
   393.2  889.92   401.6   888.8   413.1  888.66   416.6  888.66   433.1  889.16
   449.1  894.02     509  894.86     537  900.55   596.9  901.88   620.9  908.22
   640.9  908.91   660.9  915.93   688.8  929.36   776.8  966.08   820.7  988.54
#Mann= 3 , 0 , 0
       0      .1       0   401.6    .045       0   416.6     .08       0
Bank Sta=401.6,416.6
XS Rating Curve= 0 ,0
Exp/Cntr=0.3,0.1

Type RM Length L Ch R = 1 ,19009.7 ,83.5,83.4,83.3
XS GIS Cut Line= 3
     1744784.204      341888.133     1745175.321      341766.819
     1745566.439      341645.506
#Sta/Elev= 30
       0 1097.97    23.8 1086.44    47.7  1068.9    71.6 1054.37    95.4 1042.41
   119.3 1033.13   139.2 1021.97     171    1001   186.9  992.27   226.6   965.6
   258.4  948.16   306.1  926.62     330  908.59     334  907.22   345.9  907.95
   357.8  906.34   377.7  892.53   389.6  888.85     402  888.17     417  888.03
   429.4  887.66   449.3  892.94   544.7   895.5   580.5   900.4   592.4  905.68
   608.3  907.06   620.2  905.28   719.6  945.86   759.4  967.59     819 1006.54
#Mann= 3 , 0 , 0
       0      .1       0     402    .045       0     417     .08       0
Bank Sta=402,417
XS Rating Curve= 0 ,0
Exp/Cntr=0.3,0.1

Type RM Length L Ch R = 1 ,18926.3 ,66.5,66.5,66.5
XS GIS Cut Line= 3
     1744954.993      341904.859     1745032.358      341899.275
     1745665.063      341699.997
#Sta/Elev= 30
       0  993.06    50.4  960.91      62  954.76    89.6  942.67   113.5  933.93
   177.5  902.92   185.5  901.04   205.4  900.32   209.4  898.95   225.4  889.32
   245.4  886.86     247  886.87     262  886.93   269.4   887.2   289.4  895.01
   337.3  894.66   385.3  898.54   397.2  896.57   409.2     897   425.2   904.5
   453.2  907.22   469.2  917.68   477.2  921.56   489.2  930.07   541.1  951.54
   569.1  966.56     649  1017.9     673 1031.19   732.9  1060.8   740.9    1066
#Mann= 3 , 0 , 0
       0      .1       0     247    .045       0     262     .08       0
Bank Sta=247,262
XS Rating Curve= 0 ,0
Exp/Cntr=0.3,0.1

Type RM Length L Ch R = 1 ,18859.7 ,147.1,150.1,152.5
XS GIS Cut Line= 3
     1744942.841      341967.359      1745030.94      341969.425
     1745682.424      341764.234
#Sta/Elev= 30
       0  994.51    19.2  981.57    38.3  970.41    53.6   960.2    61.3  956.33
    76.6  949.29   136.1  928.51     200  901.78     212   898.8   239.9  897.44
   259.9  888.42     282  886.68   287.8  886.56     297  886.99   303.8   887.3
   319.8   891.7   423.6  895.41   427.6     896   443.6  904.48   471.6  907.66
   483.6  914.06   503.5  929.44   539.5  945.88   555.5  954.83   587.4  975.07
   607.4  985.58   679.3 1032.46   719.2 1050.39   739.2 1061.96   771.2 1083.42
#Mann= 3 , 0 , 0
       0      .1       0     282    .045       0     297     .08       0
Bank Sta=282,297
XS Rating Curve= 0 ,0
Exp/Cntr=0.3,0.1

Type RM Length L Ch R = 1 ,18709.7 ,289,300,311.5
XS GIS Cut Line= 5
     1744887.285      342074.997     1745072.821      342085.834
     1745265.922      342052.399     1745463.801      342013.137
     1745666.799       342015.97
#Sta/Elev= 30
       0 1015.78    63.3  977.78   114.7  949.02   197.8  919.19   241.8  899.76
   253.8  897.62   341.8   895.8   361.8  887.25   374.3   886.8   389.3  886.35
   393.7  886.24   405.6   886.4   425.3  890.71     453  892.19   460.9  895.65
   468.8  901.36   476.8  904.04   496.5   905.7   512.4  904.92   516.3   908.8
   528.2  927.63   536.1  933.88   567.7   943.7   591.5  956.48   623.4  982.46
     699 1034.23     707 1038.78   726.9 1045.75   754.7 1061.35   786.6 1085.03
#Mann= 3 , 0 , 0
       0      .1       0   374.3    .045       0   389.3     .08       0
Bank Sta=374.3,389.3
XS Rating Curve= 0 ,0
Exp/Cntr=0.3,0.1

Type RM Length L Ch R = 1 ,18409.7 ,300.8,300,299.2
XS GIS Cut Line= 3
     1744851.409      342219.172      1745240.97      342345.396
     1745630.531      342471.621
#Sta/Elev= 30
       0 1011.25    23.8   995.8    63.6  972.44    99.4  953.16     155  928.79
   234.6  898.74   250.5   897.1   337.9  894.05   365.8  894.88   373.7  893.04
   381.7  888.23   389.6  884.73     417  886.48   433.4  887.21   441.3  890.25
   453.2  898.02   461.2  901.04   477.1  903.45     489  903.75     493  907.21
   500.9  918.47   504.9  922.46   536.7  938.97   552.6  944.64   604.3  970.54
     648  990.55   731.5 1016.73   751.4 1019.95   771.3  1025.5     819 1033.79
#Mann= 3 , 0 , 0
       0     .08       0   381.7    .045       0     417      .1       0
Bank Sta=381.7,417
XS Rating Curve= 0 ,0
Exp/Cntr=0.3,0.1

Type RM Length L Ch R = 1 ,18109.7 ,302.5,300,298.6
XS GIS Cut Line= 3
     1744755.246      342517.875     1745148.841      342630.894
     1745542.436      342743.912
#Sta/Elev= 30
       0 1009.01    71.6  963.52   107.3  942.57   147.1  924.31   218.7  895.14
     334  892.64   361.8   893.6   369.7  892.83   377.7  888.31   385.6  883.97
   389.6  883.86   405.5  884.55   433.4  885.36   445.3  888.11   465.2  886.92
   469.1  887.71   481.1  896.11     489  899.59     497  901.23   508.9  901.01
   512.9  902.75   524.8   914.1   540.7  925.03   572.5  939.03   612.3  963.43
     664 1002.21   667.9 1005.65   679.8 1021.65   683.8 1023.91     819 1069.12
#Mann= 3 , 0 , 0
       0     .08       0   377.7    .045       0   405.5      .1       0
Bank Sta=377.7,405.5
XS Rating Curve= 0 ,0
Exp/Cntr=0.3,0.1

Type RM Length L Ch R = 1 ,17809.7 ,300.1,300,298.6
XS GIS Cut Line= 3
      1744653.09      342847.311     1745056.719      342915.762
     1745457.172      343004.229
#Sta/Elev= 30
       0  995.61    39.8  968.13    63.6  949.92    95.4  931.64   119.2  921.85
   170.9  903.87   206.7   896.5   230.5  894.05   294.1   891.4   365.7  891.28
   369.6  890.67   385.5  882.62   401.9  881.91   405.4  881.77   416.9  882.15
   441.2  885.41   477.1  887.24     493  896.35   508.9  899.62   520.9  899.79
   552.7  924.45   568.7  935.13   596.5  951.09   644.3  986.07   676.2 1007.66
   688.1    1018   723.9 1033.18   783.7 1071.38   807.6  1082.6   819.5 1089.78
#Mann= 3 , 0 , 0
       0     .08       0   401.9    .045       0   416.9      .1       0
Bank Sta=401.9,416.9
XS Rating Curve= 0 ,0
Exp/Cntr=0.3,0.1

Type RM Length L Ch R = 1 ,17509.7 ,224.5,223.9,224.2
XS GIS Cut Line= 3
     1744599.387      343144.237     1745003.075      343210.886
     1745408.201      343274.377
#Sta/Elev= 30
       0  916.96    63.6  908.25    79.4  907.67    91.4  908.82   119.2  905.16
   162.9     904   194.6  901.43   222.4  896.61   242.3  894.71   325.7  889.62
   377.4  888.81   381.4  888.01   389.3  882.59   397.2  880.89   416.7  881.99
   456.9  885.04   464.9  887.08   476.8  895.41   488.8  897.69   500.7  897.53
   528.6  920.48   560.4  931.67   592.3  947.13     644  984.41   687.8  1014.3
   723.7 1032.91   759.5  1055.5   783.4 1068.63   807.3 1079.65   819.2 1086.88
#Mann= 3 , 0 , 0
       0     .08       0   389.3    .045       0   416.7      .1       0
Bank Sta=389.3,416.7
XS Rating Curve= 0 ,0
Exp/Cntr=0.3,0.1

Type RM Length L Ch R = 1 ,17285.7 ,379.2,376.1,371
XS GIS Cut Line= 4
     1744609.507      343377.081     1744956.729      343427.428
      1745125.31      343457.686     1745265.757      343446.525
#Sta/Elev= 30
       0  949.24      16  937.12    35.9  925.05    55.8  915.12    79.7  905.11
    95.7  895.83   107.6  892.65   155.5  888.54   235.2  888.64   271.1  887.15
     291  888.08     307  883.75   326.9  882.42   337.7   879.6   338.9  879.38
   352.7  879.72   362.8   879.9   374.8  884.63   394.7  886.81   406.6  889.64
   446.4   890.4   462.4  894.36   474.3   895.9   486.3  895.18   490.3   896.5
   498.2  902.09   506.2  910.24   514.2  915.44   596.5  959.85     663  1000.7
#Mann= 3 , 0 , 0
       0     .06       0   337.7    .045       0   352.7      .1       0
Bank Sta=337.7,352.7
XS Rating Curve= 0 ,0
Exp/Cntr=0.3,0.1
